HEC-RAS study FISHINGCK.prj: FISHINGCK

--- FISHINGCK.g01 (geometry) --- (continued)

Type RM Length L Ch R = 1 ,105318  ,675.3,651.8,626.1
XS GIS Cut Line= 6
1623216.34497076388785.4963491711623381.26918159389244.661113262
1623524.94999659389644.6370193361623589.38982834389824.044140846
1623656.20596768390010.0654223411623689.87781633390103.811297834
#Sta/Elev= 30
       0  801.18    71.2  803.16   124.2  794.53   194.5  774.61   249.2  751.47
   275.2  737.02   317.7  721.21   381.5  706.29     407  696.75   581.3   689.2
     594  691.13   643.2  689.23   649.3  686.54  656.71678.3141   674.5  675.16
   751.3  675.16  762.33678.3052   780.8  685.07   806.5  683.49   830.9  687.35
     883  712.94   918.4  715.06   949.7  723.53   976.5  744.28  1044.5  788.72
    1087  810.24  1142.3  827.62    1257  829.58  1295.3  822.91  1400.8  813.85
#Mann= 9 ,-1,0
       0     .06       0      10      .1       0  424.14     .05       0
  537.89     .08       0  635.39     .07       0  656.71    .045       0
  762.33      .1       0  845.39     .07       0  952.89      .1       0
Bank Sta=656.71,762.33
XS Rating Curve= 0 ,0
Exp/Cntr(USF)=0,0
Exp/Cntr=0.3,0.1

Type RM Length L Ch R = 1 ,104666  ,580,578.1,574.6
XS GIS Cut Line= 3
1622351.02154946389349.5344835481622515.15613627389367.120332134
1623191.23431527390082.278174663
#Sta/Elev= 30
       0  757.77   129.8  715.33   220.5  692.08   244.1  687.94     347  683.81
   463.9  687.12   502.8   689.9   530.3  686.02   623.9  682.34  640.62  676.93
   661.9   674.5     761  674.54   769.5     677     781  687.38     789  691.77
   816.6  696.74   833.1  696.99   844.1   701.4   862.8  713.31   885.5  715.57
   913.8  713.82   923.4  718.78   936.4  720.86   965.2  733.65   999.1  736.21
  1021.3  739.97  1038.3  749.61  1058.7  758.41  1127.2  778.63  1149.2  781.17
#Mann= 10 ,-1,0
       0      .1       0  255.07     .05       0  395.07     .07       0
  640.62    .045       0   769.5      .1       0  825.07     .06       0
  865.07     .07       0 1005.07     .06       0 1115.07      .1       0
 1135.07     .06       0
Bank Sta=640.62,769.5
XS Rating Curve= 0 ,0
Exp/Cntr(USF)=0,0
Exp/Cntr=0.3,0.1

Type RM Length L Ch R = 1 ,104088  ,838.4,813.2,781.6
XS GIS Cut Line= 4
1622043.07246268389448.3355309861622067.86419784389754.100264573
1622596.19679291390243.4866720511623133.90880954390212.747364955
#Sta/Elev= 30
       0   788.3    40.3  787.24    72.4  778.76   128.6  748.93   151.9  731.62
   221.8   700.4   265.1   695.6   306.8  712.64     378  692.45   498.3  686.11
   516.4  690.25   560.6  683.82   669.4  684.49   681.2  682.78  688.04  677.47
   704.7  674.31   797.8   674.4   806.8  677.43   815.3   683.3   840.1  685.63
   946.1  687.58  1010.6  696.25  1151.1  704.46  1219.2  714.19  1295.3     720
  1323.3  718.88  1335.4  726.39  1383.4  733.44  1511.6  769.21  1565.5  777.43
#Mann= 11 ,-1,0
       0      .1       0  456.77     .05       0  486.77     .06       0
  596.77     .07       0  636.77    .025       0  688.04    .045       0
   806.8      .1       0  926.77     .05       0 1106.93     .06       0
 1306.93     .07       0 1496.93     .06       0
Bank Sta=688.04,806.8
XS Rating Curve= 0 ,0
Exp/Cntr(USF)=0,0
Exp/Cntr=0.3,0.1

Type RM Length L Ch R = 1 ,103275  ,803.8,816.4,831.4
XS GIS Cut Line= 3
1621620.01083624390633.0128386831622728.27129015390816.899220044
1623390.94077907390667.263506392
#Sta/Elev= 30
       0  866.27    56.9  858.08    93.4  845.97   113.6   830.9   146.1   798.2
   235.3  716.03   271.8  694.74   284.8  689.76   308.3  690.24   324.5  682.81
   340.7  681.66  350.73  675.53     361  674.25   445.8675.4477   458.3  682.59
   478.6  684.57   628.6  684.74   742.1  688.55   782.7  692.56   921.3  691.55
  1217.6  699.18  1254.5  703.15  1311.9  704.14  1451.4  722.38  1500.5  722.79
  1525.1  718.51  1582.5  714.69  1726.1  734.18  1759.2  742.96  1802.8  745.38
#Mann= 10 ,-1,0
       0      .1       0      70     .06       0     170      .1       0
     270     .07       0  350.73    .045       0   445.8     .05       0
     970     .06       0    1070     .07       0 1173.41     .08       0
 1273.41     .07       0
#XS Ineff= 2 , 0
                          799.51          717.34
Permanent Ineff=
       F       F
Bank Sta=350.73,445.8
XS Rating Curve= 0 ,0
Exp/Cntr(USF)=0,0
Exp/Cntr=0.3,0.1

Type RM Length L Ch R = 1 ,102459  ,597.2,599.1,601.3
XS GIS Cut Line= 4
1621421.48347547390949.7228190441621712.25073964391429.233745925
1622893.57826686391972.2894721951623701.71096819391903.643492732
#Sta/Elev= 30
       0  819.28      68  781.99   216.5  731.44   251.2  728.51   324.3  709.93
   370.9  702.95   487.4  697.26   508.5  690.55   541.3  693.53     565   692.6
   578.2  688.06   632.5  682.27   664.5  682.58   675.1  675.88   683.8  674.25
  780.54  675.89   798.4  684.53   824.8  686.43   908.4  683.72  1262.9  684.01
  1304.6  689.53    1393  685.86  1501.1  692.05  2064.2  697.39  2084.3  700.34
  2148.5  727.15  2172.6  733.64  2393.4   767.4  2598.1  806.52    2672  817.08
#Mann= 16 ,-1,0
       0      .1       0     240     .06       0     320     .07       0
     510     .06       0  640.78      .1       0   675.1    .045       0
  780.54      .1       0  860.78     .05       0 1190.78     .06       0
 1290.78     .07       0 1320.78     .06       0 1400.78     .07       0
 1730.78     .06       0 1790.78     .08       0 1830.78     .07       0
 2040.95      .1       0
#XS Ineff= 2 , 0
                         1022.14          704.93
Permanent Ineff=
       F       F
Bank Sta=675.1,780.54
XS Rating Curve= 0 ,0
Exp/Cntr(USF)=0,0
Exp/Cntr=0.3,0.1

Type RM Length L Ch R = 1 ,101860  ,596.4,643.3,720.5
XS GIS Cut Line= 4
1621150.58680067391465.0026803931621402.43352117391936.129735125
1622042.90578452392261.7935978431622233.96191731 392691.66989663
#Sta/Elev= 30
       0  722.68    31.2  714.09    53.9  712.91    83.5  701.27    99.3  700.54
   108.3  695.84   203.6   693.3   221.7  695.07   253.5  690.95     320  692.14
   554.1   691.2   577.4  687.05   679.7  684.95   688.7  681.81  696.19  674.68
   711.1  672.28   799.9  672.39   807.5674.7527   823.3  682.31   877.1  679.94
     979  686.73  1089.1  685.77  1240.6  693.18  1314.8  690.61  1425.4  693.08
  1455.7  697.94  1516.3  717.94  1649.7  745.34    1676  754.03  1723.2  764.37
#Mann= 12 ,-1,0
       0     .07       0     210     .08       0     320     .07       0
     510     .06       0  554.22      .1       0  696.19    .045       0
   807.5      .1       0  964.22     .06       0  984.22     .07       0
 1342.73     .06       0 1442.73     .05       0 1552.73      .1       0
#XS Ineff= 2 , 0
                         1241.18          703.13
Permanent Ineff=
       F       F
Bank Sta=696.19,807.5
XS Rating Curve= 0 ,0
Exp/Cntr(USF)=0,0
Exp/Cntr=0.3,0.1

Type RM Length L Ch R = 1 ,101216  ,144.8,141.9,138.2
XS GIS Cut Line= 4
1621049.32863551391558.9501198381621196.65365135391977.779412108
1621087.64816038 392444.860905121621084.61202951393043.553777918
#Sta/Elev= 30
       0  717.72    65.3  698.79   107.7  694.39   154.3  693.84     184  690.26
   404.9  692.55   623.4  685.84   693.3  687.24   734.3  681.88   749.8   672.8
   771.3  673.06   791.8  671.89   859.8   673.1     874  680.74   902.7  690.28
   939.3  691.04   955.3  700.78   991.3  715.55  1031.3   756.5  1047.3  769.21
  1079.3  800.18  1091.3  806.21  1115.3  811.07  1179.3  810.22  1311.3  791.94
  1343.3  781.06  1391.3  786.38  1428.3  777.71  1464.1  761.06  1522.3  743.31
#Mann= 8 ,-1,0
       0     .08       0     310     .07       0  713.98      .1       0
   771.3    .045       0   859.8     .07       0 1013.62      .1       0
 1113.62     .06       0 1413.62      .1       0
#XS Ineff= 2 , 0
          546.99  698.04
Permanent Ineff=
       F       F
Bank Sta=771.3,859.8
XS Rating Curve= 0 ,0
Exp/Cntr(USF)=0,0
Exp/Cntr=0.3,0.1

Type RM Length L Ch R = 1 ,101074  ,90.1,90,90.5
XS GIS Cut Line= 2
1621011.08953004391539.0556159381620976.47968189392976.695462272
#Sta/Elev= 30
       0  719.94    25.5  718.22    81.5   703.9   161.5  692.35   229.5  689.68
   649.7   689.4   685.7  682.18  696.45  674.16   709.7  671.22   761.7  674.15
   833.7  672.92   877.7  693.74   917.7   695.7   933.8  710.01   941.8  728.26
   949.8   736.4   969.8  745.54  1013.8  755.89  1037.8  755.28  1085.8   745.4
  1113.8  745.55  1133.8  739.92  1185.8  745.26  1217.8  738.61  1297.9  741.78
  1322.7  727.91  1341.9  723.16  1357.9  715.17    1407   717.8  1438.1  732.05
#Mann= 9 ,-1,0
       0     .07       0      10     .08       0     410     .07       0
     630      .1       0  696.45    .045       0   761.7     .08       0
     900     .07       0    1000     .06       0    1100      .1       0
Bank Sta=696.45,761.7
XS Rating Curve= 0 ,0
Exp/Cntr(USF)=0,0
Exp/Cntr=0.3,0.1

Type RM Length L Ch R = 1 ,100984  ,221.4,222.7,228.3
XS GIS Cut Line= 2
1620921.90261365391536.393319926 1620887.2927655392974.033166261
#Sta/Elev= 30
       0  720.34    36.2  709.82    84.2  703.27    96.2  698.36   152.2  691.84
   244.2  689.28   472.3  691.57   652.3  689.67   666.1  686.92   684.3  672.91
   700.3  670.85  747.07672.8663   808.4  672.45   832.4   687.1   840.4  689.39
   939.6  696.04  1036.4  697.55  1080.5  701.45  1111.5  698.17  1124.5  702.25
  1152.5  704.52  1177.9  714.58  1228.5  726.87  1268.5  729.76  1344.5  742.35
  1359.5  742.72  1400.5  737.65  1416.9  732.72  1428.6  732.59  1438.1  736.56
#Mann= 9 ,-1,0
       0      .1       0      20     .08       0     510     .07       0
     610      .1       0   684.3    .045       0  747.07     .08       0
     900     .07       0    1000     .06       0    1100      .1       0
Bank Sta=684.3,747.07
XS Rating Curve= 0 ,0
Exp/Cntr(USF)=0,0
Exp/Cntr=0.3,0.1

Type RM Length L Ch R = 1 ,100761  ,632.5,626.7,616
XS GIS Cut Line= 6
1620782.49840455 391538.22961651 1620739.6589233391832.392085927
1620712.18719347392021.0272073471620650.93994063392441.590998756
1620637.42914088392534.3621386761620580.62872955392924.388589593
#Sta/Elev= 30
       0  738.32    46.8  717.53    91.3  707.59   111.5  694.56   176.1  689.32
   386.3  690.59   580.4  687.65   600.6  681.99   620.8   682.1   635.1  673.36
   652.8  670.72   721.8  670.75   738.5673.3967   758.2  672.42   774.4  679.72
   810.8  680.91   826.9  686.71   855.2  686.52   875.4   704.7   899.7  714.35
   992.7  716.56  1037.1  735.42  1097.8  746.87  1159.1  766.79  1186.7  784.12
  1255.4  810.23  1306.1  823.33  1328.2  833.75  1356.5  841.88  1400.8  851.86
#Mann= 10 ,-1,0
       0      .1       0      10     .07       0  109.61     .08       0
  208.83     .07       0  317.27     .08       0  507.89     .07       0
   635.1    .045       0   738.5     .05       0  810.39     .07       0
 1006.64      .1       0
#XS Ineff= 2 , 0
          487.92  709.22  834.61          705.07
Permanent Ineff=
       F       F
Bank Sta=635.1,738.5
XS Rating Curve= 0 ,0
Exp/Cntr(USF)=0,0
Exp/Cntr=0.3,0.1

Type RM Length L Ch R = 1 ,100135  ,875.4,857,841.5
XS GIS Cut Line= 4
1620064.49291594391475.1728116661620065.95206541391723.728599587
1620068.81040319392402.7625413481620156.50844549392619.900706604
#Sta/Elev= 30
       0  731.88    29.4  712.49    41.4  711.02    73.4  699.81    88.5  692.63
   121.4  688.58   173.4  686.08   217.4  686.05   249.4  689.62   269.4  687.34
   281.4  682.66   289.4  682.33   413.4  683.71   521.4  678.42   569.4  680.92
   577.4  677.99  587.27  671.35   601.4  669.37   681.4  669.47   697.1  671.38
   713.4  680.59   733.3  682.01   773.3  692.09   877.4  693.81     964  700.32
  1007.2  702.18  1028.7   701.4    1046  706.88  1067.6   708.6  1161.8  717.53
#Mann= 10 ,-1,0
       0      .1       0      80     .05       0     180     .06       0
  278.56      .1       0  587.27    .045       0   697.1      .1       0
  768.56     .05       0  868.56     .06       0   967.6     .07       0
  1067.6     .06       0
#XS Ineff= 2 , 0
          249.45  708.39
Permanent Ineff=
       F       F
Bank Sta=587.27,697.1
XS Rating Curve= 0 ,0
Exp/Cntr(USF)=0,0
Exp/Cntr=0.3,0.1

Type RM Length L Ch R = 1 ,99278   ,476.7,459.7,442.8
XS GIS Cut Line= 2
1619057.78209367391517.7389161741619523.93132313392664.211369067
#Sta/Elev= 30
       0  865.02    48.7  857.67   106.7  846.17   167.1   824.7   180.1  822.65
     206  812.94   227.6  802.58   244.8  790.32   261.1  782.21   305.3  754.41
   309.6  750.62   326.9  729.06   344.1  714.58   366.2   708.5     396  690.25
   412.2  690.25   436.8  686.48   452.1  673.72  457.18  671.48   473.5  668.81
   541.2   668.9   553.5671.4518   565.7  676.93   577.3   678.4   663.7  678.37
   698.2  683.84   866.4  683.24   914.1  688.59  1095.5  691.17  1237.6   700.1
#Mann= 6 ,-1,0
       0      .1       0  457.18    .045       0   553.5      .1       0
     670     .05       0     890     .06       0    1210     .07       0
Bank Sta=457.18,553.5
XS Rating Curve= 0 ,0
Exp/Cntr(USF)=0,0
Exp/Cntr=0.3,0.1

Type RM Length L Ch R = 1 ,98818   ,506,500,490.3
XS GIS Cut Line= 6
1618425.74530001391758.4700620031618558.86970568391906.154149845
1618861.20965217392241.5632559211619099.73410951392506.176243752
1619296.93581484392724.9461474271619363.62826675392798.933532253
#Sta/Elev= 30
       0  765.95    21.5   756.8    71.1  725.95   107.9  709.32   140.9  699.18
   175.1  697.63   192.9  692.72   224.6  690.29   288.2  691.88   326.1  707.09
     350  713.04   397.8  733.62   481.5  756.52   492.8  756.61   499.4  753.14
   529.9  716.33   559.1  693.22   584.4  689.16   612.1  689.03  637.38  673.07
   654.6  668.81   735.2  668.87  747.86 673.024   756.5  676.81   784.8  678.72
   804.1  684.48   997.3  688.58  1230.6  689.76  1294.6   692.8  1400.8  702.66
#Mann= 8 ,-1,0
       0      .1       0  637.38    .045       0  747.86      .1       0
  905.39     .05       0 1046.64     .06       0 1183.52     .05       0
 1193.52     .06       0 1341.17     .07       0
Bank Sta=637.38,747.86
XS Rating Curve= 0 ,0
Exp/Cntr(USF)=0,0
Exp/Cntr=0.3,0.1

Type RM Length L Ch R = 1 ,98318   ,503.4,500,500.1
XS GIS Cut Line= 6
1617993.92201668392162.3294905131618294.45750484392417.329964757
1618566.10164659392647.8153961751618623.28952435392696.338921174
 1618761.4946285392813.6034504181619062.03011668393068.603924677
#Sta/Elev= 30
       0  868.19    65.6  858.71     113  848.06   142.2  848.52   202.2  843.67
   352.2  822.66   408.9  811.55   434.5  799.17   465.7  753.95   474.2  744.33
   545.2   689.9   573.5  689.37   585.2  691.82   595.7  689.74   630.3  690.29
   637.6  687.05  653.42  672.81   658.8  669.35   674.3  668.19   763.7  668.47
  774.04 672.877   782.4  679.11   797.7  682.88   863.2  681.69    1094  687.24
  1270.8  701.25  1303.8  707.34  1369.8  711.98  1394.5  710.91  1400.8  714.16
#Mann= 6 ,-1,0
       0      .1       0  653.42    .045       0  774.04      .1       0
  885.39     .05       0 1231.95     .06       0 1341.17     .07       0
Bank Sta=653.42,774.04
XS Rating Curve= 0 ,0
Exp/Cntr(USF)=0,0
Exp/Cntr=0.3,0.1

Type RM Length L Ch R = 1 ,97818   ,530.5,509.5,491.1
XS GIS Cut Line= 6
1617650.32198209392552.6147991721617958.09466051392798.831826419
1618512.02399884393241.9743128421618588.89097109393303.467300087
1618666.36785026393365.4488034251618744.14984693393427.674072668
#Sta/Elev= 30
       0  975.98    17.7  970.84    75.2  942.18    89.4  938.75   134.3  907.28
   166.4  894.54   198.4  874.11   211.8  872.39   223.2  866.89     288   815.4
   326.4  806.92   350.6  797.92   476.5  704.95   504.9  701.07   544.8  687.86
   564.7  685.66   584.6  688.48   613.1  680.22  628.09670.7177   647.2  666.56
   724.6  666.92   746.8  670.78   758.2  678.08   772.4  681.52  1184.5  682.79
  1286.9  686.61  1307.5  689.23  1331.7  699.99  1361.5  700.26  1400.8  723.87
#Mann= 8 ,-1,0
       0      .1       0  628.09    .045       0   746.8      .1       0
  760.39     .05       0 1016.64     .06       0 1076.64     .05       0
 1231.95     .06       0 1391.17      .1       0
Bank Sta=628.09,746.8
XS Rating Curve= 0 ,0
Exp/Cntr(USF)=0,0
Exp/Cntr=0.3,0.1

Type RM Length L Ch R = 1 ,97309   ,443.4,441.8,440
XS GIS Cut Line= 6
1617272.13966759393221.9629374011617556.68568642393307.988683985
1617649.41581592393336.0230767441617894.70108651393410.179424481
1617990.42235176393439.1180149031618612.98344259393627.334173904
#Sta/Elev= 30
       0  914.44    21.3  900.96    45.9  889.95    66.8  874.93   100.3  861.57
   167.1  817.08   233.1  791.86   259.1  773.93     278  766.67     313  745.96
   435.2  715.43   534.9  707.56   555.8  701.08   576.4  688.75   589.2  689.74
   605.9  686.28   643.5   676.5     655  668.49   672.7     666   745.5668.4037
   764.7  677.09   807.4  679.51  1134.1  680.69  1245.3  687.35  1282.9  696.83
  1314.4  697.67  1340.1  705.57  1362.3  716.48  1388.2  717.26  1400.8  727.14
#Mann= 7 ,-1,0
       0      .1       0     655    .045       0   745.5      .1       0
  912.89     .05       0 1123.52     .06       0 1221.95     .07       0
 1361.17     .06       0
Bank Sta=655,745.5
XS Rating Curve= 0 ,0
Exp/Cntr(USF)=0,0
Exp/Cntr=0.3,0.1

Type RM Length L Ch R = 1 ,96867   ,488.5,500.2,510.1
XS GIS Cut Line= 6
1617130.17135519393665.6626764921617417.47393018393741.978140661
1617686.27785452393813.3789164961617927.89876235393877.559890503
1618196.70268669393948.9606663381618484.00526169394025.276130491
#Sta/Elev= 30
       0  866.68    22.7  852.76    59.5   816.3    68.2  810.77    92.2  801.47
   126.2  797.49   146.9  789.89   187.1  764.22   226.3  748.08   279.3  733.49
     449  713.29   490.4  689.05   602.1  687.25   631.1  677.55   647.6  676.72
     661669.7806   696.8  665.75   751.1  665.78   771.5  669.75   784.2  676.57
   824.7  679.36    1016  681.73  1061.5  694.43  1094.6  694.82  1187.8  758.89
  1210.6  761.44  1230.2  776.27  1272.7  796.71  1301.6  802.21  1400.8  804.26
#Mann= 10 ,-1,0
       0      .1       0  645.39    .025       0     661    .045       0
   771.5    .025       0  845.39     .05       0 1056.64     .07       0
 1153.52     .06       0 1251.95      .1       0 1341.17     .05       0
 1361.17     .06       0
Bank Sta=661,771.5
XS Rating Curve= 0 ,0
Exp/Cntr(USF)=0,0
Exp/Cntr=0.3,0.1

Type RM Length L Ch R = 1 ,96366   ,548.5,559.8,568.7
XS GIS Cut Line= 6
 1617035.8481122394007.0333765241617123.85088894394053.761301438
1617212.19946553394098.9236126931617470.74488019394228.195991943
1617549.00751894394267.3268191911618287.25932327394636.453049446
#Sta/Elev= 30
       0  826.09    22.9  809.94   103.1  787.61   173.2  740.72   226.8  710.38
   252.4  699.56   355.3  681.67     409  688.63   444.7     680   547.6   681.4
   565.5  675.54   619.1  677.21  636.34  667.72   654.9  665.56     738667.5959
   751.6  678.04   789.1  677.95   815.9  682.16   833.8  690.82   860.6  691.37
   878.5  710.17   921.5  744.33   937.4  760.38   954.3  771.01     968  775.05
  1049.7  779.68  1151.3  793.42  1303.1  797.46  1348.1  793.91  1400.8  773.49
#Mann= 8 ,-1,0
       0      .1       0  585.42    .025       0  636.34    .045       0
     738      .1       0  800.42     .07       0  912.92      .1       0
 1133.55     .06       0 1321.21      .1       0
#XS Ineff= 2 , 0
          408.34  698.61
Permanent Ineff=
       F       F
Bank Sta=636.34,738
XS Rating Curve= 0 ,0
Exp/Cntr(USF)=0,0
Exp/Cntr=0.3,0.1

Type RM Length L Ch R = 1 ,95807   ,463.6,463.2,462.9
XS GIS Cut Line= 6
1616795.35847724394360.0348082351616952.78696814394481.479775326
1617107.43232815394600.7771089091617389.50459865394818.376083152
1617592.39887791394974.8941428231617904.47240073395215.636771576
#Sta/Elev= 30
       0  781.65    49.4  757.55    61.6  749.63    76.7  735.14    92.2  726.62
   140.6  739.05   203.8   734.7   243.3  721.27   315.2   684.9   420.1  680.81
   454.3  687.33     491  677.17   537.8  679.38   607.2  677.59   617.3  674.81
   636.1  676.46   650.4668.3033   668.8   665.5   748.1  665.57  756.91  668.34
   773.6  676.17   802.3  677.08   819.4  682.97   964.8  688.39  1015.9  701.27
  1074.8  726.31  1175.9  750.54  1287.1  785.27  1339.7  794.44  1400.8  797.48
#Mann= 7 ,-1,0
       0      .1       0   650.4    .045       0  756.91     .07       0
  875.39     .06       0 1036.64     .05       0 1201.95      .1       0
 1361.17     .05       0
#XS Ineff= 2 , 0
           448.6  691.89
Permanent Ineff=
       F       F
Bank Sta=650.4,756.91
XS Rating Curve= 0 ,0
Exp/Cntr(USF)=0,0
Exp/Cntr=0.3,0.1

Type RM Length L Ch R = 1 ,95344   ,514.2,492.2,471.1
XS GIS Cut Line= 6
1616514.06420226 394731.245697011616672.00483125394852.023670677
1617110.14207834 395187.071228941617313.69646126395342.730366427
1617390.64971943395401.5773616021617626.78474584395582.151475522
#Sta/Elev= 30
       0  867.91   113.7  840.72   187.9  805.46   239.2  808.17   274.5  800.27
   297.3  788.65   367.6  732.05   430.6  694.17   455.8  683.84   496.1   674.1
   515.7  685.81   524.6  686.39   558.8  673.94   601.8  670.76   621.1  674.97
   632.8 669.798   646.1  665.38   732.7   665.4  746.43  669.79   757.9  675.73
   788.1   675.2   807.1  681.23   843.5  684.08   921.2  683.37  1016.2  689.61
  1166.6  711.31  1226.9  714.29  1312.1  733.64  1380.6  757.29  1400.8  761.38
#Mann= 7 ,-1,0
       0      .1       0  567.89     .05       0  595.39      .1       0
   632.8    .045       0  746.43    .025       0  760.39     .06       0
  922.89     .05       0
#XS Ineff= 2 , 0
          530.27  697.71  881.09          692.53
Permanent Ineff=
       F       F
Bank Sta=632.8,746.43
XS Rating Curve= 0 ,0
Exp/Cntr(USF)=0,0
Exp/Cntr=0.3,0.1

Type RM Length L Ch R = 1 ,94851   ,483,485,487.4
XS GIS Cut Line= 6
1616180.59806702395438.6570387081616471.07911335395501.804550205
1616657.35334709395542.2992198811616742.85612884395560.886453037
1617452.07255818395715.0636381261617549.40864959395736.223372702
#Sta/Elev= 30
       0  774.01    32.3  771.44      65  750.81    73.2   749.3   132.3  779.14
   167.3  789.23   224.6   799.5   302.4  807.01   384.3  803.55   400.7  799.31
   441.6  778.79   462.1  760.32   470.2  749.78   485.4  741.78   515.6  711.17
   542.5  690.01   605.3  681.75  627.69  669.05   642.2  665.34   703.6   665.4
   716.6669.0214     724  674.52   736.3  677.48   769.1  676.51   793.6  682.81
    1027  692.81  1153.9   707.3  1326.9  719.17  1366.7  725.32  1400.8  737.97
#Mann= 7 ,-1,0
       0      .1       0  627.69    .045       0   716.6     .08       0
  800.39     .06       0  905.39     .05       0 1002.89     .07       0
 1153.52      .1       0
Bank Sta=627.69,716.6
XS Rating Curve= 0 ,0
Exp/Cntr(USF)=0,0
Exp/Cntr=0.3,0.1

Type RM Length L Ch R = 1 ,94366   ,850.6,927,997.8
XS GIS Cut Line= 6
1616311.12302026395940.4579305721616406.09199043395966.357813156
1616499.55341768395991.8475915711616674.41691311396039.537128738
1616746.77405185396059.2710131471617470.72404751396256.711563147
#Sta/Elev= 30
       0  740.76    54.9  741.16   131.2  732.37   137.7  729.08   146.1  715.76
   154.4  706.11     180  688.45   208.3  689.78   215.9  694.81   233.2  711.12
     283   707.8   299.5  700.64   328.6  678.96   345.2  675.93   353.7   667.4
   365.9  665.34   456.9  665.34   470.4 667.465     483  673.73   502.5  676.55
   763.9  688.02   870.7  704.03   912.4  717.27   979.5  731.89  1053.1  752.02
  1062.9  756.53  1105.2  787.92  1161.9  809.38  1178.5  813.08    1202   826.4
#Mann= 7 ,-1,0
       0      .1       0   353.7    .045       0   470.4     .07       0
  521.56     .08       0  571.56     .05       0  676.56     .06       0
  784.06      .1       0
Bank Sta=353.7,470.4
XS Rating Curve= 0 ,0
Exp/Cntr(USF)=0,0
Exp/Cntr=0.3,0.1

Type RM Length L Ch R = 1 ,93439   ,535.5,551.9,567.8
XS GIS Cut Line= 4
1616228.92889973 396018.00449883 1616140.7678872396157.411432689
1616077.45883229396783.4676423781615847.25435688397185.377546348
#Sta/Elev= 30
       0  709.57    21.9  701.93    55.1  686.17    83.6  682.86   130.8  684.58
   154.4  687.62   176.1  684.66   192.2  676.74   332.9  674.72   429.4  676.22
   437.5  675.23   449.5  670.34   477.7  672.58   481.7  672.13   493.7  665.68
   525.9  664.78     550  663.92   622.4  664.77   634.5  671.62   642.5  673.12
   694.8  674.07   714.9  679.14   854.6  684.86   915.3  699.67     990  713.79
  1046.4  722.05    1133  748.98  1159.4  765.22  1201.1   801.2  1257.4  825.18
#Mann= 10 ,-1,0
       0      .1       0     110     .05       0  284.94      .1       0
   525.9    .045       0   622.4      .1       0  684.94     .07       0
  784.94     .05       0  804.19     .07       0  894.19     .05       0
 1004.19      .1       0
Bank Sta=525.9,622.4
XS Rating Curve= 0 ,0
Exp/Cntr(USF)=0,0
Exp/Cntr=0.3,0.1

Type RM Length L Ch R = 1 ,92887   ,465.6,479.9,483.8
XS GIS Cut Line= 2
1615871.93872784395755.4597714251615289.09172719  397004.8123549
#Sta/Elev= 30
       0  713.45   142.1   696.1   213.1  676.42   288.1   676.2   310.7  683.46
   340.2  686.63   376.9  673.28   552.9  674.05   605.9  671.72     643  664.08
   671.3  662.62  739.24  664.14   753.1   673.2   825.4   672.4   857.5  688.12
   927.7  694.52   964.6  706.04  1020.8  711.71  1038.4  717.96    1087  751.56
  1114.3  787.51  1134.9  808.09  1166.5  822.11  1210.6  862.92  1246.7  873.33
  1264.8  887.89  1295.8  905.64  1342.9  944.04    1362  950.34  1378.6  960.87
#Mann= 5 ,-1,0
       0      .1       0     643    .045       0  739.24      .1       0
     900     .06       0    1010      .1       0
#XS Ineff= 2 , 0
          334.07  710.93
Permanent Ineff=
       F       F
Bank Sta=643,739.24
XS Rating Curve= 0 ,0
Exp/Cntr(USF)=0,0
Exp/Cntr=0.3,0.1

Type RM Length L Ch R = 1 ,92407   ,551.9,589.4,625.1
XS GIS Cut Line= 4
1615651.17124514395514.7901196461615445.26403064395775.729220078
1615081.98243292396268.8012253281614824.72592726396701.580910668
#Sta/Elev= 30
       0   740.5    93.9  687.82   155.1  673.73   256.8  672.58   293.9     683
   323.2  686.31   365.3  674.58   413.9  670.75   654.2  674.18   681.2  665.19
   730.9  661.82  821.17  665.27   830.2  673.38   850.1  676.33   888.8  694.99
   903.1   691.8   977.1  694.33  1003.3  708.53  1056.2  716.33  1112.4  760.03
    1126  774.57    1140  794.83  1156.1  807.72  1219.1  825.89  1281.6  863.59
  1328.3  877.13  1347.7  891.65    1382  904.42  1423.8  931.89  1448.3  942.12
#Mann= 9 ,-1,0
       0      .1       0     220     .05       0   342.4      .1       0
   442.4     .05       0   462.4      .1       0   681.2    .045       0
  821.17      .1       0   932.4     .07       0  954.84      .1       0
#XS Ineff= 2 , 0
          320.79     719
Permanent Ineff=
       F       F
Bank Sta=681.2,821.17
XS Rating Curve= 0 ,0
Exp/Cntr(USF)=0,0
Exp/Cntr=0.3,0.1

Type RM Length L Ch R = 1 ,91818   ,481.7,480.1,477.9
XS GIS Cut Line= 6
1615494.10910292395438.1769414251615403.42916617395480.546279252
1614954.35854201395637.7198494231614789.18301934395695.530429333
1614455.88316101 395812.185051681614175.30596626395910.385970756
#Sta/Elev= 30
       0   700.6    19.9  696.67    50.8  696.69   103.6   678.6     146  674.41
     178  673.93   196.8  683.59   221.1  686.59   239.2  682.74   256.2  673.67
   444.5  670.84   616.4  672.94   624.9  671.54   636.3  662.82   677.2  660.87
   747.8  662.83   764.7  671.48   790.2  671.91   836.8   684.6   887.1  707.28
     930  721.31   997.4  736.33  1028.8  751.83  1146.1  758.06  1204.5  791.29
  1232.8  796.21  1273.3  811.91  1307.2  813.83  1370.4   824.1  1401.3  840.85
#Mann= 7 ,-1,0
       0      .1       0  229.31     .05       0  538.37      .1       0
   636.3    .045       0   747.8      .1       0 1007.12     .06       0
 1311.65      .1       0
#XS Ineff= 2 , 0
          220.42  713.28
Permanent Ineff=
       F       F
Bank Sta=636.3,747.8
XS Rating Curve= 0 ,0
Exp/Cntr(USF)=0,0
Exp/Cntr=0.3,0.1

Type RM Length L Ch R = 1 ,91338   ,462.8,475.1,487.7
XS GIS Cut Line= 4
1615104.38279902 394885.300171981615011.17780151395094.571770163
1614385.12159182395347.807989812 1614007.0258472 395722.38656471
#Sta/Elev= 30
       0  817.34    56.1  799.63   104.3  764.14   178.7  715.53   196.5  697.09
   209.3   688.4     254  688.97   279.9  686.06   297.1  676.07   318.7  672.45
   454.1  672.98   503.5  661.67   586.2  659.88   601.7661.6953   612.1  667.95
   650.9   672.1   758.8  669.66   866.7  674.92   901.2  687.12   962.1  700.55
  1069.1  713.98    1098  721.66  1121.4  736.69    1148  742.66  1176.1  744.08
  1274.9  778.86  1350.7   786.7  1384.4  814.87  1412.6  827.92  1436.6  848.56
#Mann= 7 ,-1,0
       0      .1       0  489.09     .07       0   503.5    .045       0
   601.7      .1       0 1244.42     .05       0 1304.42     .06       0
 1436.65      .1       0
Bank Sta=503.5,601.7
XS Rating Curve= 0 ,0
Exp/Cntr(USF)=0,0
Exp/Cntr=0.3,0.1

Type RM Length L Ch R = 1 ,90863   ,154.9,222.6,307.4
XS GIS Cut Line= 4
1614857.44394951394724.1607519671614601.81760834394807.602651694
1613872.23039984394933.1858865571613672.97608133395070.393801487
#Sta/Elev= 30
       0   826.4    30.9  810.83    47.7  797.92   131.8  741.71   144.1  730.55
   156.8  715.05   190.7  689.54     198  687.68     216  688.97   242.4  684.13
   282.8  681.26   295.4  676.63   343.7   669.3  358.45  661.08   380.2  659.03
   453.3  661.02   493.9  661.43   527.4  666.42   550.7  665.22   587.2  671.53
   652.1  669.47   757.7  671.38   879.5   670.2   960.6  676.74  1062.8  699.18
  1168.2  718.27  1198.5  732.52  1212.6  736.72  1224.5  745.45  1251.1  754.46
#Mann= 3 ,-1,0
       0      .1       0  358.45    .045       0   453.3      .1       0
Bank Sta=358.45,453.3
XS Rating Curve= 0 ,0
Exp/Cntr(USF)=0,0
Exp/Cntr=0.3,0.1

Type RM Length L Ch R = 1 ,90640   ,235.8,195,138.1
XS GIS Cut Line= 3
1614863.65053141394711.547955183 1614597.5542305394799.108885707
1613338.10916885394491.568934329
#Sta/Elev= 30
       0  837.14    19.4  822.57    96.4  780.02   151.1  738.54   209.5  689.32
   285.7  681.07   368.1  677.67   442.7   663.2   504.9661.4194   705.7  658.62
  739.64  661.47   763.4  670.62   845.7  668.68   932.1   674.3   999.2  670.03
  1066.6  670.54  1090.9  674.48  1113.4   670.8  1166.6  670.54  1195.7  676.69
  1261.6  676.89  1286.3  684.72  1339.2  691.74  1393.3  692.93  1428.5  703.25
  1459.2   700.3  1467.5  703.11  1508.6  731.78    1541  758.04  1576.6  778.85
#Mann= 3 ,-1,0
       0      .1       0   504.9    .045       0  739.64      .1       0
#XS Ineff= 2 , 0
           328.2  691.72  941.96           692.3
Permanent Ineff=
       F       F
Bank Sta=504.9,739.64
XS Rating Curve= 0 ,0
Exp/Cntr(USF)=0,0
Exp/Cntr=0.3,0.1

Type RM Length L Ch R = 1 ,90445   ,285.8,268.1,257.7
XS GIS Cut Line= 3
1614876.64649523394634.1536037411614538.11199974394672.771728148
1613395.61309172394394.468315179
#Sta/Elev= 30
       0  856.68    56.9  842.81   161.6  806.38   188.8  790.24     222  762.61
   238.1  754.18   302.6   708.2   340.7  693.39   392.2  682.83   466.3  672.98
   585.7  671.75   626.9  667.88   643.3  661.99   685.2659.9952   729.8  658.56
     798660.0911   845.1  670.16   971.6  674.77  1005.6  671.34    1051  672.91
  1186.8   670.5  1209.9   674.7  1232.1  672.98  1249.7  679.14  1281.5  680.89
  1297.9  679.12  1330.9  685.53  1380.3  687.55    1442  701.54  1516.6  748.36
#Mann= 5 ,-1,0
       0      .1       0  590.73    .025       0  660.73      .1       0
   685.2    .045       0     798      .1       0
#XS Ineff= 2 , 0
          468.57  690.04 1051.08          701.31
Permanent Ineff=
       F       F
Bank Sta=685.2,798
XS Rating Curve= 0 ,0
Exp/Cntr(USF)=0,0
Exp/Cntr=0.3,0.1

Type RM Length L Ch R = 1 ,90177   ,585.4,634.1,680.9
XS GIS Cut Line= 4
1614900.25187136394585.2898523941614323.71445602394354.240408697
   1613555.14774394367.2669632061613400.00242371394328.506851574
#Sta/Elev= 30
       0  856.88    51.9  841.51    69.1  834.08    86.3  831.72   152.6  812.02
   228.5  784.67   301.8  762.24   379.1  742.66   391.4  742.46     556  708.08
   581.9  695.86   612.1  689.69   640.7  677.59   692.7  671.77   760.7  671.53
   804.7     664   840.7  667.02   868.7  660.91   907.1660.7384   968.8  657.69
   996.8  657.78 1007.61  660.83  1024.8  671.13  1245.1  667.35  1324.8  674.99
  1356.8  681.62  1390.2   683.6  1417.7  689.78  1467.1  706.97  1549.7  752.47
#Mann= 5 ,-1,0
       0      .1       0  741.11    .025       0  841.11      .1       0
   907.1    .045       0 1007.61      .1       0
#XS Ineff= 2 , 0
                         1300.72          694.34
Permanent Ineff=
       F       F
Bank Sta=907.1,1007.61
XS Rating Curve= 0 ,0
Exp/Cntr(USF)=0,0
Exp/Cntr=0.3,0.1

Type RM Length L Ch R = 1 ,89543   ,724.7,725,723.3
XS GIS Cut Line= 6
1614698.75085837394322.7395819881614556.95192936394290.679278657
1614458.81465845394235.001896575 1613965.7713532 393476.47191757
1613912.12447887393393.9373057341613803.76544363393227.231274322
#Sta/Elev= 30
       0  733.07    23.2  727.08   314.5  680.63   394.9  674.73     576   674.4
   630.1  668.17   661.9  670.64  683.67  661.25   690.5  658.36   714.4   657.5
   762.3   657.7   776.4   661.3   790.7  669.45   828.3  683.34   895.7  690.13
   943.4   700.4   961.7  720.17   970.3  732.45   995.8  757.37  1011.8  768.87
  1048.3  809.18  1091.3  826.01  1146.7  860.33  1167.6  880.44    1201  902.54
  1220.1  911.69  1250.8  952.21  1285.5  973.54  1320.3  972.67  1460.2  946.21
#Mann= 3 ,-1,0
       0      .1       0  683.67    .045       0   776.4      .1       0
Bank Sta=683.67,776.4
XS Rating Curve= 0 ,0
Exp/Cntr(USF)=0,0
Exp/Cntr=0.3,0.1

Type RM Length L Ch R = 1 ,88818   ,498.4,500,501.5
XS GIS Cut Line= 6
1615213.46202642394053.634106845   1614654.68985393215.470756918
1614600.08300383393134.1831898391614544.55621201393051.504549429
1614488.62062834392968.3472354261614242.85668418392994.824872762
#Sta/Elev= 30
       0  805.18    82.5  759.23     146  729.05   260.9  697.05   345.2  684.77
   442.3  675.68   635.9  674.61   650.3  671.84  667.65661.1111   679.2  657.19
   708.5  656.94   736.9   660.3   766.8  657.78   797.9  661.07   818.6  670.65
   838.3  674.67   878.9  700.83   890.2  711.09   924.3  750.47   947.9   766.1
   996.4  806.93    1055  827.76    1088  844.45  1105.2  848.84  1160.3  854.56
  1304.9  841.67  1349.8  844.73  1442.4  838.95  1494.8  828.42  1552.3  822.02
#Mann= 3 ,-1,0
       0      .1       0  667.65    .045       0   797.9      .1       0
Bank Sta=667.65,797.9
XS Rating Curve= 0 ,0
Exp/Cntr(USF)=0,0
Exp/Cntr=0.3,0.1

Type RM Length L Ch R = 1 ,88318   ,494.3,491.9,490.7
XS GIS Cut Line= 6
1615601.84806067393770.9073100841615202.45647101 393135.63364625
1615014.50737184392836.6814882611614962.11410393392753.345368832
1614793.37625243 392745.796827511614395.23466025392883.549504757
#Sta/Elev= 30
       0  820.53    26.4  809.25    54.8  804.37   116.2  763.18   201.2  728.11
   347.7  685.18     499  672.09   623.8  673.08   649.6  668.26   658.6  659.64
   673.1  656.66   758.8  659.58   815.3  671.15   853.3  693.84   900.5  728.54
   930.9  746.58    1047  793.62  1084.8  797.34    1132  789.03  1183.2  785.68
    1202  780.06    1264  793.83  1344.1  804.81  1389.7  802.72  1461.1  806.96
  1537.3  796.96  1579.6  812.71  1697.9  838.48  1723.5  838.49  1792.2  825.42
#Mann= 3 ,-1,0
       0      .1       0   658.6    .045       0   758.8      .1       0
Bank Sta=658.6,758.8
XS Rating Curve= 0 ,0
Exp/Cntr(USF)=0,0
Exp/Cntr=0.3,0.1

Type RM Length L Ch R = 1 ,87826   ,625.2,543,454.6
XS GIS Cut Line= 6
 1616021.9157901393507.2300159191615510.85266508392716.682865992
 1615275.0016015392672.9905426651615095.45865351392669.552557424
1614860.04869126392703.9002577511614428.57055159392862.601383924
#Sta/Elev= 30
       0  882.86    17.8  872.71      41  868.56   106.7  823.47   154.3   811.7
   191.5  794.08   276.2  742.43   323.3  704.59   337.4  697.13   363.5   689.4
   426.9  678.82   594.3  672.69     628  667.87   638.9659.2123   729.4  656.62
  745.21  659.28     768  667.51   936.9  680.23  1151.9  685.36  1336.3     705
  1444.2  726.83  1481.6  743.09  1578.6  767.18  1652.3  792.26  1769.3  799.17
    1829  794.75  1882.9  812.78  1990.9  838.08  2020.8  838.98  2058.6  831.13
#Mann= 4 ,-1,0
       0      .1       0   638.9    .045       0  745.21    .025       0
  817.89      .1       0
Bank Sta=638.9,745.21
XS Rating Curve= 0 ,0
Exp/Cntr(USF)=0,0
Exp/Cntr=0.3,0.1

Type RM Length L Ch R = 1 ,87283   ,479.7,465.1,447
XS GIS Cut Line= 6
 1616220.3532069392035.9481739171615614.10573174392596.067788578
1615523.50191033392626.9420706551615066.64455633392640.152017987
1614853.65747197392687.0578710791614459.55961808392843.159360669
#Sta/Elev= 30
       0  989.25    27.6  975.87    49.3  960.31    83.4  950.27   119.5  932.08
   190.9  887.05   234.5  869.35   289.7  826.02   348.9  807.24   365.2  793.02
     436   714.6   447.8  704.86   490.5  690.89   512.9  679.62   602.1  674.44
   648.7659.0154   670.2  656.38  740.34  659.02   759.2  670.25   781.8  678.74
  1163.8   684.2    1385  705.68  1473.1  725.55  1521.7  743.84  1596.4  764.37
  1641.1  780.97  1817.5  792.96  1903.5  819.66  1976.6  836.61  2020.3  838.06
#Mann= 3 ,-1,0
       0      .1       0   648.7    .045       0  740.34      .1       0
Bank Sta=648.7,740.34
XS Rating Curve= 0 ,0
Exp/Cntr(USF)=0,0
Exp/Cntr=0.3,0.1

Type RM Length L Ch R = 1 ,86818   ,514.3,500,479.4
XS GIS Cut Line= 6
1615681.45190409391580.7712704241615222.94921218 392476.93023926
1615177.62843667 392562.560973511615046.77239917392614.337772846
  1614835.705236392676.2930295021614416.39898801392848.797605753
#Sta/Elev= 30
       0  996.86    58.1  987.71    98.6  962.44   134.7  948.43     157  927.05
   229.7  880.57   280.2  835.29   315.9  820.01   341.2  794.89   381.7  767.09
   426.6  755.61   471.5  709.23   480.5  703.39   552.4   682.5   628.8  674.15
  656.78659.7616   682.7  656.38   731.8  656.49   750.1  659.76   763.6  661.29
     804  679.98  1082.4  683.31  1220.3  696.64  1305.4   710.1  1492.4  770.99
  1628.1  782.48  1736.8   814.3  1835.8  838.65  1861.7  839.15  1917.6  827.96
#Mann= 5 ,-1,0
       0      .1       0  635.39    .025       0  650.39      .1       0
  656.78    .045       0   750.1      .1       0
Bank Sta=656.78,750.1
XS Rating Curve= 0 ,0
Exp/Cntr(USF)=0,0
Exp/Cntr=0.3,0.1

Type RM Length L Ch R = 1 ,86318   ,524.3,500,461.2
XS GIS Cut Line= 6
1614983.51366742391360.5512384181614906.30089533   391930.737434
1614861.01128776392265.1849278361614822.22101101392551.633173838
1614723.42987001392644.940401927  1614360.261305392833.121456012
#Sta/Elev= 30
       0  983.95    49.2  975.35   185.7  925.23   242.2  912.97   274.5  900.51
   302.7   885.1   339.1  836.71   378.9  816.74   395.6  803.51   403.6   795.4
   415.7  776.76   484.4   706.6   544.9  683.82   629.7   675.2   649.9  668.52
   657.9  662.26   682.2  656.38   754.8  656.47  774.87662.4708   819.4  679.26
  1021.2  680.75  1081.8  685.24  1194.8  701.83  1280.5  727.71  1331.4   736.4
  1391.1  770.09  1454.2  795.48  1608.3   825.8  1648.6  827.34  1746.9  815.28
#Mann= 3 ,-1,0
       0      .1       0   657.9    .045       0  774.87      .1       0
Bank Sta=657.9,774.87
XS Rating Curve= 0 ,0
Exp/Cntr(USF)=0,0
Exp/Cntr=0.3,0.1

Type RM Length L Ch R = 1 ,85818   ,472.7,470.1,473.4
XS GIS Cut Line= 6
1614184.77871634391401.3887551721614244.08371584 391591.16659084
1614408.60044718392117.6219027491614543.29013842392548.629242837
1614570.70806259392644.0119260851614283.90023726392832.657218084
#Sta/Elev= 30
       0  998.28    45.2  987.18    74.5  971.87   116.4  959.74   175.1  925.82
   288.3   883.9   351.1  840.87   401.4  820.62   439.1  790.03   493.5  762.11
   531.3   724.6   543.9  705.32   560.5  691.82   627.6  668.26   637.6  660.67
   665.4  654.88     787  655.12     797  660.71   820.5  676.79   967.2  675.98
  1074.8  682.34  1210.2  707.62  1226.8  714.15  1301.2  760.33  1361.8  777.16
  1404.8  797.92  1459.4  809.34  1500.6  811.95  1538.9  806.93  1644.5  782.27
#Mann= 4 ,-1,0
       0      .1       0  567.89    .025       0   637.6    .045       0
     797      .1       0
#XS Ineff= 2 , 0
                          826.46          694.69
Permanent Ineff=
       F       F
Bank Sta=637.6,797
XS Rating Curve= 0 ,0
Exp/Cntr(USF)=0,0
Exp/Cntr=0.3,0.1

Type RM Length L Ch R = 1 ,85348   ,528.2,565.3,593.3
XS GIS Cut Line= 6
1613712.11612513391534.3611561071613740.15871997391630.104731024
 1614043.4802918392484.9156854461614108.79446564392668.983886853
1614141.97451739392762.4902615251614083.55239014392886.704251946
#Sta/Elev= 30
       0  899.39    14.8  891.44    35.6  887.48    48.1  881.53    98.5  849.45
   216.9  832.37   246.7  826.96   267.9  819.74   280.6  813.32   330.3  774.71
   365.5  761.13   446.1  712.16   555.9  683.85   575.5  671.19   598.9  661.36
   634.6  658.77   645.6  654.53   726.3  654.31   745.2658.8395   760.2  667.48
   951.2  679.63  1014.9  696.74  1036.1  699.89  1104.4  732.48  1154.9  764.58
  1214.4  783.11  1256.8  803.61  1364.4  831.53  1400.8  838.01  1438.6  837.93
#Mann= 3 ,-1,0
       0      .1       0   634.6    .045       0   745.2      .1       0
Bank Sta=634.6,745.2
XS Rating Curve= 0 ,0
Exp/Cntr(USF)=0,0
Exp/Cntr=0.3,0.1

Type RM Length L Ch R = 1 ,84783   ,499.1,510.7,522
XS GIS Cut Line= 4
1613620.47325833391562.3081993221613428.41676965392063.232621844
1613363.02422155392309.9739577341613149.54144854392853.937141515
#Sta/Elev= 30
       0  894.71    36.7  877.46    83.8  843.78   113.8  827.44   146.3  817.54
   263.7  742.51   306.5  722.05   389.1  701.75   591.6  670.24     604   665.3
   628.9  665.45   643.4657.1276   674.4  653.91   740.6  653.97   748.9  657.22
   757.1  666.27   777.8  677.64   914.8  706.55  1000.8  738.39    1048   760.3
  1065.2  763.62  1086.7  772.92    1120  797.94  1181.7  824.39  1215.8  848.34
  1237.2  867.04  1284.4  888.98  1325.3  912.43  1361.7  946.47  1376.1  955.78
#Mann= 4 ,-1,0
       0      .1       0  616.48     .07       0   643.4    .045       0
   748.9      .1       0
Bank Sta=643.4,748.9
XS Rating Curve= 0 ,0
Exp/Cntr(USF)=0,0
Exp/Cntr=0.3,0.1

Type RM Length L Ch R = 1 ,84272   ,397.6,409.4,425.5
XS GIS Cut Line= 6
1613243.33930553 391388.165106041613106.76838445391652.201323372
1613019.19113178391821.5182419541612898.59196352392054.674927872
1612691.13371702392455.7604117961612599.78711494392632.363076952
#Sta/Elev= 30
       0  789.57    41.8  791.42      68  785.53   106.6  768.43   174.8   719.8
   198.6  710.22   234.2  707.73     255  695.89   294.3  702.32   536.9  678.69
   603.9  676.04     626  665.47   637.9  664.03   646.3  657.48   662.4  653.84
   743.5  654.02  749.39  657.51   759.5  665.05   842.6  675.74   903.8  697.48
  1004.7  764.25  1060.5  807.97  1115.7  830.88  1172.1   876.7  1207.7  887.56
  1260.8  911.75  1306.4  946.41  1346.9  957.13    1374  974.16  1400.8  979.99
#Mann= 3 ,-1,0
       0      .1       0   646.3    .045       0  749.39      .1       0
Bank Sta=646.3,749.39
XS Rating Curve= 0 ,0
Exp/Cntr(USF)=0,0
Exp/Cntr=0.3,0.1

Type RM Length L Ch R = 1 ,83863   ,533.3,521.9,509.8
XS GIS Cut Line= 6
1613086.99894963391229.6360647711612885.73360414391448.403015676
1612578.94386338391781.8734773431612273.21153522392114.193022686
1612338.55490846392290.0312536841612444.44708513392483.055145848
#Sta/Elev= 30
       0  780.96      72  765.35    96.3  754.71   221.4  716.19   270.3  711.89
   287.8  713.19   465.1  689.67   498.6  688.98   642.3  676.82   663.7  667.19
   680.7  666.22     692  655.89   714.6  653.75     790   653.9  798.77     656
   807.7  665.53   810.9  666.49   898.7  676.36   924.1  682.32   992.1  710.56
  1011.9  729.35  1032.2  756.13  1096.8  816.74  1139.3  832.76  1170.4  854.49
  1181.7  856.06    1202  853.96  1315.4  881.79    1397  892.71  1609.7  938.54
#Mann= 4 ,-1,0
       0      .1       0  680.39    .025       0     692    .045       0
  798.77      .1       0
Bank Sta=692,798.77
XS Rating Curve= 0 ,0
Exp/Cntr(USF)=0,0
Exp/Cntr=0.3,0.1

Type RM Length L Ch R = 1 ,83341   ,511.7,506.7,503.3
XS GIS Cut Line= 6
1612504.91960039390859.1138492731612013.60004497391737.709533027
1611995.77166856391838.7332810971612064.42244989391996.920628777
1612216.62654181392232.520879349 1612365.9490778392455.425617269
#Sta/Elev= 30
       0  729.77      52  750.65    88.7  752.84     162  732.64   432.4  683.23
   560.8  680.75   624.9  674.36   642.4  666.61   652.4  657.02   671.8  652.91
   734.9  652.97  746.85  656.92   753.2  660.05   789.4  654.13   803.6  657.56
   815.8  666.02   848.1  670.43   895.3  700.07   973.2  725.48  1041.4  732.26
  1109.2  731.81  1137.4  736.92  1246.4  764.47  1391.7  791.55  1435.9  811.59
  1495.5  829.52  1567.6  841.89    1697  879.94  1776.8  891.65  1830.5  904.58
#Mann= 5 ,-1,0
       0      .1       0  567.89    .025       0   652.4    .045       0
  746.85    .025       0  760.39      .1       0
Bank Sta=652.4,746.85
XS Rating Curve= 0 ,0
Exp/Cntr(USF)=0,0
Exp/Cntr=0.3,0.1

Type RM Length L Ch R = 1 ,82834   ,631.4,515.9,411.6
XS GIS Cut Line= 6
1611988.40105938390635.7964559771611644.49886004391386.130585221
1611650.84760063391486.172707972 1611718.6119008391623.369940144
1611974.27379105391991.0460420671612327.00963413392476.667446149
#Sta/Elev= 30
       0  780.32    31.6  775.76    66.8  753.93   103.4  744.41   163.6   756.6
   227.1  751.66   317.6   717.6     388  704.49   471.1  682.63   572.8  673.08
   594.8  664.23  603.61  655.04     696  652.91   715.1655.0121   726.8  664.78
   770.8  662.98   788.4  670.14   819.2  675.41  1215.8  683.59  1293.6  688.62
  1508.9  717.66  1647.5  756.51  1671.9  769.49    1712  779.46  1772.8  809.48
  1806.6  819.98  1875.2  832.14  1922.7  835.83    2060  877.31  2126.7   886.3
#Mann= 5 ,-1,0
       0      .1       0  603.61    .045       0   715.1      .1       0
  995.63     .05       0 1298.75      .1       0
Bank Sta=603.61,715.1
XS Rating Curve= 0 ,0
Exp/Cntr(USF)=0,0
Exp/Cntr=0.3,0.1

Type RM Length L Ch R = 1 ,82318   ,526.8,500,472
XS GIS Cut Line= 6
1610674.03705017391345.9420156781611489.82970992391471.448326334
1611572.67173584391511.5886660071611678.68300676391618.834842592
1611816.53738984391777.193121672 1612322.9369676392444.053008422
#Sta/Elev= 30
       0 1014.49   103.3  980.72   159.9  950.14   184.2  930.51   212.5  916.73
   236.8  908.39   253.8  906.85     338  870.63   382.5  839.18   418.9  820.38
   443.2  794.78   471.6  772.22   540.4     700   601.1  678.93  633.01659.8219
   657.7  652.96   714.4  652.75   754.9  654.67   762.9  659.81   803.4  677.72
  1224.3  681.94  1316.4   688.5  1491.5  712.52  1583.3  734.81  1721.6  780.03
  1807.8  819.96  1882.1  834.03  1932.7  839.25  2056.7  877.66  2115.6     887
#Mann= 5 ,-1,0
       0      .1       0  633.01    .045       0   762.9      .1       0
  895.39     .05       0  1328.2      .1       0
Bank Sta=633.01,762.9
XS Rating Curve= 0 ,0
Exp/Cntr(USF)=0,0
Exp/Cntr=0.3,0.1

Type RM Length L Ch R = 1 ,81818   ,504.3,500,493.1
XS GIS Cut Line= 6
1610764.30885126392153.400374502  1611724.116971391849.930837095
1611839.25420792391892.741118923  1611974.388124392021.821569428
1612159.83361925392242.8686995061612325.77685693392458.496549085
#Sta/Elev= 30
       0 1039.03    50.1 1006.91     155   979.2   214.1  951.31   255.7  905.59
     348  844.73     369  823.72   385.8  817.25   452.9  761.75   469.7   737.4
   493.8     723     520  700.28   637.5  666.23  661.67655.4382   682.6  651.69
  754.95655.4144   767.5  661.51   792.7  661.07   855.6  676.16  1036.7   679.2
  1141.7  689.18  1313.2  719.42  1406.2  749.31    1440   766.9  1475.7  776.68
  1539.2  808.12  1574.2  819.85  1684.1  836.05  1815.2  877.28    1877  887.45
#Mann= 5 ,-1,0
       0      .1       0  661.67    .045       0  754.95      .1       0
 1036.64     .05       0 1139.48      .1       0
#XS Ineff= 2 , 0
                          826.23          700.83
Permanent Ineff=
       F       F
Bank Sta=661.67,754.95
XS Rating Curve= 0 ,0
Exp/Cntr(USF)=0,0
Exp/Cntr=0.3,0.1

Type RM Length L Ch R = 1 ,81318   ,488.3,500,514.5
XS GIS Cut Line= 6
1610919.53327835392691.4363719221611370.21774442392504.566010758
1611938.89574093392268.7708786731612029.82764567392231.070166677
1612187.55338009392347.4928340911612339.63673735392510.808780417
#Sta/Elev= 30
       0  985.65   100.2  946.16   132.9  920.51   185.1   892.1   212.8  881.45
   234.5  878.16   269.1  856.82   305.7   843.3   334.1  823.24   381.7  800.81
   520.9  706.08   593.9  672.43   644.6  662.88  653.78653.9251   667.5  651.25
  771.45653.9105   780.1  661.44   788.7  663.49   866.7  667.38  1013.9  693.44
  1044.2  694.52  1057.2  701.74  1126.1  718.94  1161.1  732.47  1243.8   772.6
  1294.3  790.25    1349   819.9  1404.8  830.86  1551.4  876.97  1621.2  889.26
#Mann= 3 ,-1,0
       0      .1       0  653.78    .045       0  771.45      .1       0
Bank Sta=653.78,771.45
XS Rating Curve= 0 ,0
Exp/Cntr(USF)=0,0
Exp/Cntr=0.3,0.1

Type RM Length L Ch R = 1 ,80818   ,501.8,500,497.5
XS GIS Cut Line= 6
1611023.37854309392999.3320815861611220.01824167392969.913505256
1611666.61052434392903.0999905911611765.50993285392888.304088429
  1612018.939216392850.3891379981612408.74191409392792.072325513
#Sta/Elev= 30
       0  923.12    41.2  899.61    69.5   880.5   101.9  868.02   158.5  821.45
   178.7   813.8     203  800.62   235.3  775.94   284.6  750.53   352.6  705.33
   380.9  699.41   433.5  683.16   579.1  662.74   634.9  662.26   643.8  660.16
  654.18651.9934     664  650.41  753.14651.9317   773.2  666.39   797.5  677.89
     846  695.83   878.4  697.39   910.8  711.59   991.7  763.34  1032.1   783.3
  1072.5  810.26  1141.3  828.88  1246.5  878.85  1343.6  912.81  1400.8  941.72
#Mann= 3 ,-1,0
       0      .1       0  654.18    .045       0  753.14      .1       0
Bank Sta=654.18,753.14
XS Rating Curve= 0 ,0
Exp/Cntr(USF)=0,0
Exp/Cntr=0.3,0.1
