HEC-RAS study FISHINGCK.prj: FISHINGCK

--- FISHINGCK.g01 (geometry) --- (continued)

Type RM Length L Ch R = 1 ,32818   ,495.2,500,507.4
XS GIS Cut Line= 6
1594220.39705725406328.0705159161594306.77910234406377.670810416
1594478.18853642406476.0925295951594562.19919518 406524.33127825
1595348.78390808406975.9835901711595435.16628125407025.583556592
#Sta/Elev= 30
       0  737.78    41.2  711.25   267.2  650.85   345.6  650.11     424  631.42
   524.6  630.26     567  640.89   643.6  624.99  657.54613.8596   738.5  611.88
     748  613.91   764.9  625.69   783.8  625.15   817.6   638.7   848.4  638.59
   867.4  646.58   964.9  661.11  1021.1  689.87  1063.8  702.46  1088.2  718.54
  1107.7  742.04  1148.7  776.43  1180.5  790.12  1198.9     809  1245.4   843.9
  1263.5  849.38  1301.2  871.21  1333.3  897.52    1388  911.34  1400.8  919.17
#Mann= 10 ,-1,0
       0      .1       0      10     .05       0  347.27      .1       0
  367.27     .05       0  575.39      .1       0  657.54    .045       0
     748      .1       0  760.39     .06       0  800.39     .07       0
  912.89      .1       0
#XS Ineff= 2 , 0
          564.82  659.59
Permanent Ineff=
       F       F
Bank Sta=657.54,748
XS Rating Curve= 0 ,0
Exp/Cntr(USF)=0,0
Exp/Cntr=0.3,0.1

Type RM Length L Ch R = 1 ,32318   ,498.2,499.5,501.5
XS GIS Cut Line= 6
1594016.33972259406673.3437755111594096.05052118406733.118262261
1594174.10253042406794.3740452531594470.32995634407026.857832253
1594607.99601959407134.8996109221595119.63377585407536.440146416
#Sta/Elev= 30
       0  746.68    39.7  718.06    85.3  701.24   110.7  696.88   135.3  686.24
   176.4  661.28   290.1  628.45   442.1  626.12   491.2  638.28   519.8  628.96
   642.9  624.64  668.12612.8922   679.4  611.88  753.15612.8689     766  621.45
   811.5  636.03   845.7  638.07   862.8  646.06   902.1  648.93     928  655.73
  1004.8  690.36  1065.8  706.73  1096.4   726.1    1122  756.65  1170.5   794.7
  1192.9  821.04  1232.5  850.69  1255.9  857.87  1294.6  862.35  1400.8  860.22
#Mann= 7 ,-1,0
       0      .1       0  377.29     .05       0  517.91      .1       0
  668.12    .045       0  753.15      .1       0  855.41     .06       0
  895.41      .1       0
#XS Ineff= 2 , 0
           486.1  659.09
Permanent Ineff=
       T       F
Bank Sta=668.12,753.15
XS Rating Curve= 0 ,0
Exp/Cntr(USF)=0,0
Exp/Cntr=0.3,0.1

Type RM Length L Ch R = 1 ,31819   ,506,500.5,492.9
XS GIS Cut Line= 6
1593704.99454476407040.9844444251594082.54497075407349.823721752
1594151.53695875407403.5752546791594284.19056484407517.721023753
1594411.75330184407618.6814517531594796.93953934407919.290758669
#Sta/Elev= 30
       0  696.55   122.9  681.05   184.9  665.17     372  633.28   456.7  630.49
   485.7   637.4   516.5  627.98   591.9  627.88   625.4  625.27   655.5  618.65
   664.2  613.41   678.4  611.88  753.28613.3777   775.7  624.21   818.9  625.49
   860.4  629.89   877.1   637.1   903.2   636.9   928.6  651.46   938.8   654.4
  1009.9  654.24  1042.7  676.45  1078.3  694.47  1097.8  699.09  1125.4     712
  1162.8  744.25  1230.8  786.51  1282.1  807.07  1309.2  813.61  1401.5  822.04
#Mann= 7 ,-1,0
       0      .1       0  169.56     .05       0  547.78      .1       0
   664.2    .045       0  753.28      .1       0  800.24     .07       0
  1036.8      .1       0
#XS Ineff= 2 , 0
          482.16  661.94
Permanent Ineff=
       F       F
Bank Sta=664.2,753.28
XS Rating Curve= 0 ,0
Exp/Cntr(USF)=0,0
Exp/Cntr=0.3,0.1

Type RM Length L Ch R = 1 ,31318   ,468.3,472.6,477.7
XS GIS Cut Line= 6
1593372.70255843   407524.9975841593456.90711442407578.210404083
1593785.14070992407785.6351860911594070.44591358407965.932397678
1594305.55896042408114.5101845121594556.85242109408273.313672677
#Sta/Elev= 30
       0  726.11    68.8  698.27   109.4  685.49   133.9  681.64   183.8  667.87
   283.7  649.52   396.8  640.56   413.9  634.26   428.4   636.3   451.6  634.55
   491.4  627.97   631.3  626.39  656.61614.1602     669  611.88  757.46614.0389
   770.4  625.41   784.8  631.79     872  633.75   907.8   644.3   978.8  687.87
  1054.5  691.47  1073.4  695.38  1086.5  702.03  1097.1  713.28  1106.5   718.7
  1121.3  754.26  1139.7  771.73  1149.1  789.33  1153.2  792.07  1400.8  812.27
#Mann= 10 ,-1,0
       0      .1       0      80     .05       0  198.83      .1       0
  497.89     .05       0  656.61    .045       0  757.46    .025       0
  780.39      .1       0  865.39     .06       0  895.39     .03       0
 1046.64      .1       0
#XS Ineff= 2 , 0
          429.64  643.63
Permanent Ineff=
       F       F
Bank Sta=656.61,757.46
XS Rating Curve= 0 ,0
Exp/Cntr(USF)=0,0
Exp/Cntr=0.3,0.1

Type RM Length L Ch R = 1 ,30845   ,528.8,571.3,608.4
XS GIS Cut Line= 4
1593357.63537309407829.5950286841593650.73284954408250.786957796
 1593874.3553686408424.4743512451594503.97216985 408326.77519243
#Sta/Elev= 30
       0  676.12      70  662.52   144.9  649.11   207.4  632.85   222.9  634.64
   271.6  628.21   383.7  626.72   456.8  628.59     525  625.33  546.61  615.04
   566.7  611.88   635.1   611.9   643.6  615.08     679  629.41   703.5  630.14
   747.9  627.18   780.5  635.99   836.3  640.21   911.4  668.12   947.8  687.84
     960  690.22  1020.7  692.46  1040.9  703.71    1049   715.5  1065.2  747.38
  1069.3  752.88  1095.6  763.92  1150.2  772.76  1283.8  785.27  1433.4  804.24
#Mann= 8 ,-1,0
       0     .05       0      70      .1       0     140     .05       0
     320     .08       0     430      .1       0  546.61    .045       0
   643.6     .07       0  743.14      .1       0
#XS Ineff= 2 , 0
          220.48   642.4
Permanent Ineff=
       F       F
Bank Sta=546.61,643.6
XS Rating Curve= 0 ,0
Exp/Cntr(USF)=0,0
Exp/Cntr=0.3,0.1

Type RM Length L Ch R = 1 ,30274   ,446,456.1,465.6
XS GIS Cut Line= 6
1593099.31561881407882.7880458451593147.36276681407979.166462011
1593186.27476248408075.669549844 1593207.1917154408172.487597681
1593216.99222073408268.865685753 1593318.8371614409270.341045014
#Sta/Elev= 30
       0  752.22    46.6  723.09    64.5  714.32   104.8  703.44   195.4  664.19
   234.2  649.51   282.2  637.45   301.5  629.21   326.9  633.44   351.1   627.1
   411.4  625.06   523.9  627.48   560.5  626.36   604.4  621.82   628.5  624.26
   636.5  623.19   654.6   613.1   668.7  611.88   754.5613.0095   765.2   618.7
   773.2  628.57   782.5  632.48   829.5  635.61  1090.8  638.66  1132.8  657.58
  1171.3  662.62  1207.4  660.97  1275.8  650.81  1314.7  650.57  1414.3  653.29
#Mann= 12 ,-1,0
       0      .1       0   320.8     .05       0  427.67     .08       0
  618.92    .025       0   654.6    .045       0   754.5     .05       0
  918.92      .1       0 1016.42     .07       0 1117.05     .06       0
 1215.48     .05       0  1314.7     .07       0 1414.31     .06       0
Bank Sta=654.6,754.5
XS Rating Curve= 0 ,0
Exp/Cntr(USF)=0,0
Exp/Cntr=0.3,0.1

Type RM Length L Ch R = 1 ,29818   ,457.5,464.9,472.3
XS GIS Cut Line= 6
1592826.59078975407886.4532259261592819.89460893408085.326843917
1592816.30570534408183.7666076721592812.33196001408280.611558333
1592807.58754693408374.2662266791592740.64575167409284.699117094
#Sta/Elev= 30
       0  775.21    22.1  769.33    58.1  751.72   111.4  758.38   154.2  758.48
   182.2   754.1   206.2  742.77   246.2  717.29   258.2  715.86   286.3  705.74
     333  677.43   362.3  665.12   418.4  632.64   438.4  632.11   462.4     624
   626.8  624.16   634.8  621.73   642.9  614.35   658.9  611.88   751.2   611.9
   759.7 614.341   779.2   626.6   803.3  628.94   931.7   631.3  1112.1  630.59
  1148.2   628.4  1200.4  631.67  1224.4  638.23  1268.6   638.9  1401.1  669.18
#Mann= 11 ,-1,0
       0      .1       0  595.69    .025       0   642.9    .045       0
   759.7      .1       0  790.69     .05       0  993.19     .07       0
 1086.94     .05       0 1183.82     .07       0 1282.26     .06       0
 1301.47      .1       0 1381.47     .06       0
#XS Ineff= 2 , 0
                          1016.1          650.18
Permanent Ineff=
       F       F
Bank Sta=642.9,759.7
XS Rating Curve= 0 ,0
Exp/Cntr(USF)=0,0
Exp/Cntr=0.3,0.1

Type RM Length L Ch R = 1 ,29353   ,546,535.1,523.7
XS GIS Cut Line= 6
 1592467.5070302407836.8708050351592448.25674063407934.602236877
1592410.05865429408128.5326232861592373.21883295408315.563745285
 1592235.2220617409016.1650343791592216.21488188409113.546401287
#Sta/Elev= 30
       0  724.47    81.2  743.32   105.7  741.76   150.5  726.15   183.1  718.66
   199.4  711.63   215.7  710.09   252.4  691.71   289.1  680.73   366.6  668.31
   456.3  661.06   468.5  656.29   492.8  637.32   505.2  631.69   525.6  632.42
     550  622.14   627.5  621.67   639.7  615.04     656   611.5   745.1  611.28
  766.34  615.02   778.3  622.69   831.3  623.68   876.2  628.94  1067.8  630.23
  1116.7  632.97  1153.4  630.57  1181.9  637.71  1230.9  642.34  1301.2  660.79
#Mann= 6 ,-1,0
       0      .1       0   639.7    .045       0  766.34     .05       0
 1096.64     .07       0 1163.52     .06       0 1261.95      .1       0
Bank Sta=639.7,766.34
XS Rating Curve= 0 ,0
Exp/Cntr(USF)=0,0
Exp/Cntr=0.3,0.1

Type RM Length L Ch R = 1 ,28818   ,487.4,500,515.5
XS GIS Cut Line= 6
 1591805.6866636407785.0144524281591801.25130501408272.884867758
1591800.45603101408360.3814119251591799.77394576408435.378309175
1591798.18339776408610.3710694161591794.75984818408986.917888507
#Sta/Elev= 30
       0  697.59    27.5  691.32   155.4   670.7   195.5  666.54   227.5   666.4
   271.5  662.94   351.5  651.35   403.5  649.54   451.5   645.1   543.5  648.72
     551   645.9   559.5  637.64   567.5  633.09   607.5  631.63   647.5  610.67
   659.5  609.66   755.6  610.71   771.6  618.26   779.6  619.92   795.6  618.08
   968.3  630.71  1011.6  629.81  1035.6  635.17  1047.6  641.08  1079.6  663.56
  1107.6  694.08  1139.6  720.79  1147.6  724.34  1171.6  728.04    1202  741.41
#Mann= 8 ,-1,0
       0      .1       0  208.83     .05       0  497.89      .1       0
   647.5    .045       0   755.6    .025       0  790.39     .05       0
  992.89     .06       0 1086.64      .1       0
Bank Sta=647.5,755.6
XS Rating Curve= 0 ,0
Exp/Cntr(USF)=0,0
Exp/Cntr=0.3,0.1

Type RM Length L Ch R = 1 ,28318   ,494.7,500,510.5
XS GIS Cut Line= 6
1591512.06585975407765.1145578321591477.80805425407858.994291335
1591444.50529934407952.7319647521591413.11133325408046.186174169
1591385.53625718408139.0724713361591222.65534934408729.518140838
#Sta/Elev= 30
       0  669.89    80.6  662.26   220.3  660.73     338  647.12   371.5  644.56
   471.1   626.6   483.5  629.22   537.5  630.02   554.1  633.63   583.1  631.05
   603.9  621.31   637.1  622.94   655.9  611.61     671  609.62   757.4  609.65
     764611.5349   794.8  631.17   807.2  635.47     833  637.44   865.3  636.02
   881.9  643.42   906.8  661.61   923.4  678.79   933.9  682.26     940  686.59
   963.1   716.9   977.3  721.61   998.9  734.79  1002.2  736.92  1007.4  744.17
#Mann= 8 ,-1,0
       0     .05       0     338      .1       0  548.64    .025       0
   655.9    .045       0     764     .07       0  826.14    .025       0
  856.14     .06       0  953.64      .1       0
#XS Ineff= 2 , 0
          529.03  641.92
Permanent Ineff=
       F       F
Bank Sta=655.9,764
XS Rating Curve= 0 ,0
Exp/Cntr(USF)=0,0
Exp/Cntr=0.3,0.1

Type RM Length L Ch R = 1 ,27818   ,490.9,500,506.8
XS GIS Cut Line= 6
1591127.70737651407583.9508781731591009.75944968407856.815489918
 1590971.3218625407945.7388685051590934.12377417408031.793486416
1590869.64785326408180.9546054151590728.29610184408507.961825415
#Sta/Elev= 30
       0  662.25    79.6  653.59   140.1  649.66   222.2  652.63   301.2  650.31
   331.8  647.04   379.8   635.8   405.9  632.82   482.9   631.3     493  633.03
   508.2  631.51   519.2  633.04   532.6  631.03   562.8  631.41   597.6  622.41
   610.7  621.54   632.5  610.98   645.6  609.53   727.3  609.57   732.9610.9814
   745.8  620.36   806.8  628.16     846  636.18   885.5  652.58   902.7  663.26
     907  664.37   928.8  666.36   981.1  663.17   998.6  670.17  1006.6   675.2
#Mann= 7 ,-1,0
       0     .05       0  547.89    .025       0   632.5    .045       0
   732.9      .1       0  760.39    .025       0  875.39     .06       0
  885.39     .07       0
Bank Sta=632.5,732.9
XS Rating Curve= 0 ,0
Exp/Cntr(USF)=0,0
Exp/Cntr=0.3,0.1

Type RM Length L Ch R = 1 ,27318   ,595.3,581.8,567.3
XS GIS Cut Line= 6
1590741.75604868407414.8337623331590599.55226484407676.179696336
1590367.87326625408065.602145836  1590334.171562408132.845449671
1590303.65751542408216.2908208371590280.03748393408309.497327343
#Sta/Elev= 30
       0  657.65    52.7  655.32   130.1  654.09   192.8   649.6   215.7   649.6
   233.9  647.86   261.4  643.01   297.4  638.32   320.4  632.67     353  628.59
   385.2  627.56   427.6  628.56   455.3  630.19   464.9  632.45   478.6  630.14
   524.7   627.9   560.2  624.07   609.5  623.22     618  622.18   621.4  620.79
   632.8  611.31   637.5  609.92   646.8  609.53   730.8  609.55   751.7611.3303
   798.7  619.18   838.3  628.22   893.7  631.54   917.9  634.81  1010.9  658.53
#Mann= 9 ,-1,0
       0     .05       0  129.72     .06       0  317.53     .05       0
  528.17      .1       0   632.8    .045       0   751.7      .1       0
  770.67     .06       0  885.89     .05       0  984.74     .07       0
Bank Sta=632.8,751.7
XS Rating Curve= 0 ,0
Exp/Cntr(USF)=0,0
Exp/Cntr=0.3,0.1

Type RM Length L Ch R = 1 ,26736   ,858.8,766.4,686.7
XS GIS Cut Line= 3
1590048.43173703407263.9353265031589740.77040824408197.044638807
 1589827.7932444408461.444720603
#Sta/Elev= 30
       0  668.95    19.7  663.91    55.4  659.59   110.1  648.44   178.1  648.05
   218.2  640.15   244.9  638.77   367.1   625.7   392.3  632.24   400.8  631.27
   417.6   625.4   421.8  625.03   489.2  623.54   552.4  619.56   590.3  620.53
   607.1  617.96  617.88  610.35     624  608.51   632.4  608.19   712.4  608.26
   720.9  610.33   741.9  626.03   746.1  627.67     932  629.71     970  634.02
  1019.9  644.76  1073.5  650.46  1146.2  660.78  1188.3  663.59  1260.9  663.56
#Mann= 11 ,-1,0
       0      .1       0      40     .05       0     140     .06       0
     350      .1       0     560    .025       0  617.88    .045       0
   720.9    .025       0     760     .05       0     970     .06       0
 1072.52     .07       0 1162.52     .06       0
Bank Sta=617.88,720.9
XS Rating Curve= 0 ,0
Exp/Cntr(USF)=0,0
Exp/Cntr=0.3,0.1

Type RM Length L Ch R = 1 ,25970   ,688.4,651.9,611.7
XS GIS Cut Line= 3
 1589006.4302524408166.6722359781589511.00343543408349.369612891
1589791.11462841408513.587622831
#Sta/Elev= 30
       0  778.52    10.3  770.03    31.6  756.23    65.6  743.37    82.6  732.93
    95.4  718.62   108.1  697.93   112.4  693.22   129.4  679.87   154.9  654.93
   163.4  648.67   176.2  633.13   201.7  629.26   235.8  627.11   248.5  621.74
     257  614.58     264  611.24   278.3  607.41   376.2  607.42   388.9  608.58
   393.2  611.18   393.2  611.19   421.3  621.99   439.8  632.84     491  642.05
     508  643.58   598.3  645.19   690.9   659.2   715.1  661.38   861.3  663.49
#Mann= 8 ,-1,0
       0      .1       0     110     .06       0     220      .1       0
     264    .045       0   393.2    .025       0     430      .1       0
  596.63     .05       0  756.63     .07       0
Bank Sta=264,393.2
XS Rating Curve= 0 ,0
Exp/Cntr(USF)=0,0
Exp/Cntr=0.3,0.1

Type RM Length L Ch R = 1 ,25318   ,392.9,375.7,362.9
XS GIS Cut Line= 6
1588712.90413526409096.9868940861589183.85824583408969.552437678
 1589340.7171841 408927.108624921589437.24586242  408900.9889265
 1589684.6003546408834.0579580071590022.22376481408708.202082319
#Sta/Elev= 30
       0  928.39    69.6     911    98.6  906.92   123.5   898.1   140.1  884.31
   166.1  869.11   206.4   839.7   235.4  830.69   254.1  808.55   305.8  760.75
   326.5   748.1   355.6  734.27   404.1  693.29   446.7  663.41   487.9  647.53
   546.2  642.13   558.6  638.62   575.2  630.01   612.5  626.92   633.2  619.13
   643.3609.2271   658.1  606.12   740.9  606.16   753.4  609.32   778.2  622.17
   840.4  629.69   873.8  643.82   898.4  649.42  1253.7   651.4    1367  668.24
#Mann= 9 ,-1,0
       0      .1       0  517.89     .06       0  615.39      .1       0
   643.3    .045       0   753.4    .025       0  820.39     .06       0
  922.89     .07       0 1186.64     .06       0 1336.64     .07       0
Bank Sta=643.3,753.4
XS Rating Curve= 0 ,0
Exp/Cntr(USF)=0,0
Exp/Cntr=0.3,0.1

Type RM Length L Ch R = 1 ,24942   ,200.5,181.2,165.8
XS GIS Cut Line= 4
1589135.00028253409393.8052840161589381.20216274409348.863670961
1589668.43768965 409165.189252391589959.58118292408834.966095596
#Sta/Elev= 30
       0  754.76    29.6  742.15    49.9  720.81    67.4  699.82    90.6  682.23
   102.8  669.06     119   666.3   163.8  642.03   180.8  635.88   208.5  630.53
   228.8  630.88     241  628.12   253.7  631.84   263.2   630.9   324.9  614.73
   334.4   608.5   343.9  606.14   419.9  606.12  433.46  608.62   458.2  619.55
   491.1  621.13   529.1   626.7   571.8  642.69   594.3  648.11   681.4  649.19
     748  645.64   775.7  641.98   850.8  641.28   899.2  642.93  1031.5  652.21
#Mann= 8 ,-1,0
       0     .06       0     180      .1       0   334.4    .045       0
  433.46      .1       0  590.27     .06       0  641.21     .07       0
  791.21     .06       0  861.21     .07       0
#XS Ineff= 2 , 0
          254.32  640.33
Permanent Ineff=
       F       F
Bank Sta=334.4,433.46
XS Rating Curve= 0 ,0
Exp/Cntr(USF)=0,0
Exp/Cntr=0.3,0.1

Type RM Length L Ch R = 1 ,24761   ,120.8,126.6,120.6
XS GIS Cut Line= 3
1589312.31462427409768.8162792181589443.53788415409596.349955334
1589987.68343387 408931.68894829
#Sta/Elev= 30
       0  642.59    31.5  641.48      80  636.75   100.9  635.41   302.3  630.39
   331.3  628.45   337.6  625.91   350.6  613.86   358.1608.9554   362.9     607
   369.2  606.11   413.1     606   457.6   606.2   464.3  606.91   468.4609.0248
   482.8   617.1   492.7  618.83   518.3  625.82   552.4   629.7   593.8  633.05
   615.4  635.71   643.4  637.47   653.3  637.13   707.6  639.25   743.8  642.09
   826.5  650.22   845.2  650.14   893.3  647.44   912.2  647.49  1075.7  653.74
#Mann= 8 ,-1,0
       0     .08       0     140     .07       0   358.1    .045       0
   468.4     .08       0  526.71     .07       0  906.71     .06       0
  936.71     .08       0 1036.71     .07       0
#XS Ineff= 2 , 0
          262.76  639.15
Permanent Ineff=
       F       F
Bank Sta=358.1,468.4
XS Rating Curve= 0 ,0
Exp/Cntr(USF)=0,0
Exp/Cntr=0.3,0.1

Type RM Length L Ch R = 1 ,24635   ,199.8,202.5,203.9
XS GIS Cut Line= 3
1589388.74869843409836.5159800771589500.14362926 409705.90946199
1590044.28917898409041.248454946
#Sta/Elev= 30
       0  647.42    63.1  646.22     110  643.76   126.1  644.72     147   643.9
   241.1  637.17   249.4  634.93   274.9  624.46   303.4   618.1   319.9608.0293
   323.3  606.42   329.5  605.97   417.1  605.97     431608.1075   443.1  617.01
   447.4  618.76   462.9  619.25   473.3  620.96   506.3  632.93   525.2  635.35
   569.4  636.19   597.3  638.24   657.8  646.99   692.8  648.82   752.4  647.38
   814.5  647.72   834.9  649.29   853.6  648.04   904.1  652.15  1030.7  655.89
#Mann= 14 ,-1,0
       0     .08       0      20     .07       0     110     .08       0
  171.66     .06       0  241.66     .07       0   319.9    .045       0
     431     .08       0  621.66     .07       0  641.66     .06       0
  751.66     .07       0  801.66     .06       0  871.66     .07       0
  951.66     .06       0 1001.66     .07       0
Bank Sta=319.9,431
XS Rating Curve= 0 ,0
Exp/Cntr(USF)=0,0
Exp/Cntr=0.3,0.1

Type RM Length L Ch R = 1 ,24432   ,1608,1626.7,1606.9
XS GIS Cut Line= 4
1589560.86151555409931.9817103251589923.89602769409499.827085534
1590102.75438643409157.0866705681590248.79928014409093.589074429
#Sta/Elev= 30
       0  644.36    24.6  641.34    51.5  633.17   171.7  626.86   187.3  625.04
     212  618.47   231.9  616.18   234.7  615.08   241.4  607.92   251.8     606
   286.6  605.94   328.4  605.97  341.61  607.93   359.5  614.71   375.4  618.47
   402.2  618.68     459   624.4   467.5  626.85   490.2  639.66     513  641.35
   546.1  646.85   593.7  648.28   679.7  647.39   694.5  643.49   706.3  646.08
     717  646.91   741.9  646.37   766.6     644   890.2  654.68  1110.3  667.01
#Mann= 9 ,-1,0
       0     .06       0     220      .1       0     230     .06       0
   241.4    .045       0  341.61     .06       0     360      .1       0
     520     .07       0   724.4      .1       0   834.4     .06       0
Bank Sta=241.4,341.61
XS Rating Curve= 0 ,0
Exp/Cntr(USF)=0,0
Exp/Cntr=0.3,0.1

Type RM Length L Ch R = 1 ,22805   ,633.4,641.8,651.7
XS GIS Cut Line= 2
1590752.55441881409982.7767051391591431.82336008409168.384372332
#Sta/Elev= 30
       0  668.83    38.2  662.15    60.2  661.85   107.1  647.35   134.8  640.93
   164.4  640.22   190.4  636.09   249.1  632.79     430  626.75   555.1  623.87
   594.8  616.37   620.4  614.58     628  606.87   642.5  605.28     717  605.35
  727.64606.8767   754.9  619.24   785.1  621.42   810.7  636.06   862.4  678.09
   867.4  684.92     878  705.08   893.6  723.11   909.2  733.81   924.3  738.89
     930  742.49   950.9  763.83  1017.2  794.59  1034.2  798.82  1060.5  802.06
#Mann= 7 ,-1,0
       0     .06       0     170     .05       0     200     .06       0
     300     .05       0     430      .1       0     628    .045       0
  727.64      .1       0
Bank Sta=628,727.64
XS Rating Curve= 0 ,0
Exp/Cntr(USF)=0,0
Exp/Cntr=0.3,0.1

Type RM Length L Ch R = 1 ,22164   ,757.7,761.9,765.9
XS GIS Cut Line= 2
1591099.47935897410377.6333032561591966.13663612 409631.20593738
#Sta/Elev= 30
       0  734.31    21.1  726.44    55.1  704.24    83.5  689.31   137.4  670.24
   291.2  648.99   381.7  655.61   510.4  636.26   633.7  633.87   655.4  621.01
   673.4  616.31   686.9607.3613   697.7  605.12   789.7  605.18   800.4  607.33
   820.9  620.97   840.8  622.63   871.9  633.73     889  635.95   920.2  658.57
   961.6  675.41   988.5  697.21  1014.4  725.68  1047.8  737.77  1061.9   757.5
  1077.8  773.48  1090.4  800.67    1096  807.68  1111.1  812.63  1143.8  817.24
#Mann= 8 ,-1,0
       0      .1       0      50     .06       0     230     .05       0
     360     .06       0     500     .05       0     620      .1       0
   686.9    .045       0   800.4      .1       0
Bank Sta=686.9,800.4
XS Rating Curve= 0 ,0
Exp/Cntr(USF)=0,0
Exp/Cntr=0.3,0.1

Type RM Length L Ch R = 1 ,21402   ,631,641.9,651.5
XS GIS Cut Line= 2
1591481.68640245410979.4776492051592448.53527234410253.088601876
#Sta/Elev= 30
       0  713.79    58.1  691.32   118.1   677.5   135.2  671.34   155.2  670.93
   238.1  655.21   329.5  664.47   352.4  663.35   404.5  654.94   518.4  664.51
   628.4  662.81   660.9  653.11   692.3  637.03   738.5  621.37  766.01  607.39
     778  605.13   878.6  605.12   895.4 607.414   910.6  617.43     938  619.69
   958.6  626.33   978.6  624.05  1008.7  629.33  1040.9  644.92    1077  672.14
  1098.7  682.54  1110.3  691.17  1158.8  698.93  1188.8  712.42  1209.3  717.22
#Mann= 6 ,-1,0
       0      .1       0     110     .06       0     230      .1       0
  766.01    .045       0   895.4    .025       0     970      .1       0
Bank Sta=766.01,895.4
XS Rating Curve= 0 ,0
Exp/Cntr(USF)=0,0
Exp/Cntr=0.3,0.1

Type RM Length L Ch R = 1 ,20760   ,508.8,535.1,566.5
XS GIS Cut Line= 2
1591697.33108082411426.3471924231592904.63977328410810.168897103
#Sta/Elev= 30
       0  706.33      45  686.18   196.7  659.31   317.5  655.74   344.4  647.16
   364.7   635.1   483.6  661.86   510.6  658.89   573.5  665.14   667.8  660.88
   687.3  655.21   737.8  629.24     789  618.31   815.1  617.88   827.6606.6872
   833.9  605.12   930.4606.6445   968.7  618.12   977.6   624.7  1009.1  631.01
  1080.9  636.52  1166.3  671.38  1211.2  717.68  1269.5   741.9    1283  755.84
  1296.5  777.75  1305.5  787.31  1326.5  798.34  1341.4  812.94  1355.5  820.31
#Mann= 5 ,-1,0
       0      .1       0      80     .06       0     190      .1       0
   827.6    .045       0   930.4      .1       0
Bank Sta=827.6,930.4
XS Rating Curve= 0 ,0
Exp/Cntr(USF)=0,0
Exp/Cntr=0.3,0.1

Type RM Length L Ch R = 1 ,20225   ,602,637.6,677.3
XS GIS Cut Line= 2
1591689.17899188411505.8026321681593125.50412414411538.670484165
#Sta/Elev= 30
       0  727.12      91  691.32     159   674.3     175  673.62     207  667.31
     255  662.28     323  664.29   416.3  660.48   563.1  642.43   662.7  633.84
   867.2  629.13   887.2  619.03   899.2  615.42   909.2   607.9   919.2  605.12
  1019.2  605.12  1030.5607.8463  1043.2  618.33  1047.2  619.18  1103.2  621.24
  1119.2  624.95  1147.2  643.17  1179.2  670.41  1211.3  692.56  1263.3  721.88
  1327.3  746.17    1355  765.02  1391.3   784.5  1411.3  787.49  1436.7  795.28
#Mann= 5 ,-1,0
       0      .1       0      80     .06       0     280      .1       0
   909.2    .045       0  1030.5      .1       0
#XS Ineff= 2 , 0
          863.13  636.96
Permanent Ineff=
       F       F
Bank Sta=909.2,1030.5
XS Rating Curve= 0 ,0
Exp/Cntr(USF)=0,0
Exp/Cntr=0.3,0.1

Type RM Length L Ch R = 1 ,19587   ,657.6,660.3,663.2
XS GIS Cut Line= 2
1591729.49493448411590.3242340131593146.09935554412691.397275902
#Sta/Elev= 30
       0  723.64      54   709.1    89.4  696.55   226.2  671.75   348.4  665.68
   388.2  661.17     488  639.68   550.7  630.72   661.9  623.97   707.5  626.62
   714.1  623.72   727.8  608.99  731.36  606.73     743  604.97   824.4     605
   835.7 606.625   854.4  607.11     870  610.24   892.8  612.29   910.2  610.32
   978.3  619.88  1150.8  622.36  1462.4  637.38  1535.3  642.88  1634.6  663.62
  1651.1  665.32  1673.9  673.36  1733.7  688.08  1750.4  696.33  1794.2  723.44
#Mann= 10 ,-1,0
       0      .1       0     170     .06       0     300      .1       0
  731.36    .045       0   835.7    .025       0     870      .1       0
    1030     .05       0    1350     .06       0    1420     .05       0
    1670      .1       0
#XS Ineff= 2 , 0
                         1252.88          642.89
Permanent Ineff=
       F       F
Bank Sta=731.36,835.7
XS Rating Curve= 0 ,0
Exp/Cntr(USF)=0,0
Exp/Cntr=0.3,0.1

Type RM Length L Ch R = 1 ,18927   ,764.2,878.2,965.6
XS GIS Cut Line= 3
1591699.77475778411696.8896058311591552.54978833412263.692426729
1592422.29807631412995.396182681
#Sta/Elev= 30
       0  702.29    24.4  688.08    81.4  669.29   123.6  665.14   185.6  662.76
   278.3  666.93   462.5   666.8   585.6   664.5   634.2  659.51   684.4  646.31
   731.4  656.42   785.8  658.99     813  664.74   867.3  664.34   898.7   656.9
   924.8  656.51   953.5  649.19   978.4  637.41     997  623.02  1008.9  617.56
 1025.29605.8889  1034.3  604.97  1167.9  605.86  1183.4  615.51  1233.2  614.28
  1311.6  622.09  1426.2  625.35  1506.5  630.29  1630.6   655.7  1722.2  665.94
#Mann= 8 ,-1,0
       0      .1       0      30     .06       0     140      .1       0
 1025.29    .045       0  1167.9      .1       0 1255.61     .05       0
 1435.61     .06       0 1585.61     .05       0
Bank Sta=1025.29,1167.9
XS Rating Curve= 0 ,0
Exp/Cntr(USF)=0,0
Exp/Cntr=0.3,0.1

Type RM Length L Ch R = 1 ,18049   ,819.7,844.9,862.6
XS GIS Cut Line= 4
 1591645.6720954 411704.474663711591476.30091516412342.051280572
1591291.65382335412443.3093631731590956.89597073412979.058356121
#Sta/Elev= 30
       0  685.61    47.1  669.21    62.1  668.39    78.7  662.85   107.7   660.5
   148.5  663.72   219.4  662.32   273.2  666.92     356  662.91     447  665.82
   496.7  660.08   546.4   658.2   659.7  660.63   828.7  633.47   937.6  631.12
   960.8  620.11   984.9  616.13   995.7  606.86  1012.8  604.97 1130.48  606.81
  1145.3  616.33  1201.9  624.87  1239.6  640.04  1322.3  643.09  1402.1  663.88
  1418.9  672.59  1457.2  699.58  1461.3  705.51  1473.3  730.27    1502   759.3
#Mann= 8 ,-1,0
       0     .06       0     130      .1       0  960.28    .025       0
   995.7    .045       0 1130.48     .06       0 1190.28     .07       0
 1280.28     .05       0 1420.28      .1       0
Bank Sta=995.7,1130.48
XS Rating Curve= 0 ,0
Exp/Cntr(USF)=0,0
Exp/Cntr=0.3,0.1

Type RM Length L Ch R = 1 ,17204   ,588.4,630.5,668
XS GIS Cut Line= 2
1591416.53896478411339.7601050891590272.25078416412281.160310427
#Sta/Elev= 30
       0  760.85    57.5  737.69    88.6  729.82   148.6  684.92   183.8  674.36
   202.6  673.31   249.2  655.46   285.4  655.17   332.1   640.8   350.4  639.21
   399.4  656.51   451.2  661.34   492.5  660.21   549.6  653.28   627.3  660.58
   685.7  652.27   731.6  649.02   891.5   625.2   938.1  622.69   964.2  615.22
   989.9  615.13  1000.2  606.96  1014.9  604.97 1124.72606.9811  1145.3  614.12
    1223  621.45  1264.4  635.03  1387.6  656.27  1447.3  676.37  1481.8  697.95
#Mann= 10 ,-1,0
       0      .1       0     150     .06       0     190      .1       0
     450     .07       0     460      .1       0  1000.2    .045       0
 1124.72     .05       0    1210     .06       0    1230     .05       0
    1340      .1       0
Bank Sta=1000.2,1124.72
XS Rating Curve= 0 ,0
Exp/Cntr(USF)=0,0
Exp/Cntr=0.3,0.1

Type RM Length L Ch R = 1 ,16573   ,903.8,842.1,793.3
XS GIS Cut Line= 4
1591181.18891345411120.6410917771590913.37678607411388.453219158
 1589809.6662005411473.6661687791589647.35582027411648.149827527
#Sta/Elev= 30
       0  767.65    17.7  755.45    86.4  730.89   176.9  676.62   303.3  667.58
   412.1  666.21   596.7  657.49   632.2  647.55   660.8  626.76   677.9   621.1
     713  616.56   801.3  615.74  816.72606.2509   829.3  604.97   957.7  606.27
   965.7  612.13   981.8  615.49  1057.8   617.4  1102.2  621.09  1266.9  623.47
  1439.2  620.99  1493.9  623.29  1531.3  636.52  1598.9  637.53  1627.6  650.95
  1653.6  652.11  1669.9  660.73    1687  663.95  1705.3  672.01    1724  684.01
#Mann= 14 ,-1,0
       0      .1       0     160     .06       0     290      .1       0
  518.74     .06       0  618.74      .1       0  816.72    .045       0
   957.7      .1       0 1008.74     .05       0 1108.74     .06       0
 1208.74     .05       0 1408.74     .08       0 1515.74     .07       0
 1565.74     .06       0 1695.74      .1       0
Bank Sta=816.72,957.7
XS Rating Curve= 0 ,0
Exp/Cntr(USF)=0,0
Exp/Cntr=0.3,0.1

Type RM Length L Ch R = 1 ,15731   ,524.5,530.8,541.5
XS GIS Cut Line= 2
1590333.03986842410346.6072313041589603.24925467411589.725141164
#Sta/Elev= 30
       0  757.71    54.7  733.71    71.8  720.06    86.8   705.6   108.9  689.42
   159.9  659.12   178.5   652.6   207.3  647.04   224.9  641.34   257.3   637.8
   271.3   631.2     310  618.22  330.13606.0411   345.5  604.94  438.25605.9807
   447.5  612.25   452.2  613.37   499.6  613.27   577.8  617.25     800  622.31
  1089.3  621.17  1197.4  622.83  1223.7  627.97  1244.2  636.65  1314.9  637.23
  1352.3  653.74  1379.8  654.46  1393.2  661.72  1407.9   664.1  1441.5  682.01
#Mann= 15 ,-1,0
       0      .1       0     120     .06       0     230     .05       0
     290     .06       0  330.13    .045       0  438.25    .025       0
     460     .05       0     580     .06       0     690     .05       0
     800     .06       0     870     .08       0    1030     .05       0
    1070     .08       0    1150     .07       0    1380     .06       0
Bank Sta=330.13,438.25
XS Rating Curve= 0 ,0
Exp/Cntr(USF)=0,0
Exp/Cntr=0.3,0.1

Type RM Length L Ch R = 1 ,15200   ,433.3,431.5,428.6
XS GIS Cut Line= 2
1589887.24308635410166.636850863 1589085.7085182411155.686386789
#Sta/Elev= 30
       0  737.89    17.7  723.95    49.4  694.16    84.8  671.97    94.6  659.93
   105.4  639.68   114.5  632.66     123  630.86   208.4  629.43     240  622.92
     288  615.16   310.7   606.8   326.8  604.94   411.6  604.95   422.9606.8804
   447.2  620.42   460.7  622.04   608.5  619.21   697.5  621.16   910.8  619.35
   996.1  623.44  1034.2  635.07  1067.2  640.64  1087.1  646.51  1135.1  649.87
  1150.6  653.19  1217.9  671.58  1248.4  688.42    1269  689.73  1273.1   692.2
#Mann= 12 ,-1,0
       0      .1       0     110     .08       0     150     .07       0
     240    .025       0     310     .07       0   310.7    .045       0
   422.9    .025       0     460     .07       0     490     .05       0
     930     .06       0    1120      .1       0    1250     .06       0
Bank Sta=310.7,422.9
XS Rating Curve= 0 ,0
Exp/Cntr(USF)=0,0
Exp/Cntr=0.3,0.1

Type RM Length L Ch R = 1 ,14769   ,162.1,165.4,169.3
XS GIS Cut Line= 3
1589486.10347957409955.5283554681588921.93256018410735.453306575
1588825.98077413411009.514588787
#Sta/Elev= 30
       0  647.44    70.4  647.45     100  645.72   105.8  644.43   116.7  638.57
   129.6  637.27   139.9  632.48   183.9  630.56   231.3  621.44   262.8  617.29
     280  606.33   287.6  604.94   401.1  604.94  407.55  606.36   415.9  612.99
   434.7  620.98   440.4  621.69   849.7  619.25   914.6  620.19   921.7  621.99
   939.2  630.23   980.6  630.76  1044.3  659.03  1052.8  659.63  1069.7   655.2
  1101.2  661.67  1159.5  667.11  1184.1  672.09  1226.5   686.5    1253  689.81
#Mann= 10 ,-1,0
       0     .06       0     120     .07       0     150      .1       0
     250    .025       0     280    .045       0  407.55     .05       0
     850     .06       0 1002.59     .08       0 1072.59     .05       0
 1182.59     .06       0
#XS Ineff= 2 , 0
                          811.07          641.55
Permanent Ineff=
       F       F
Bank Sta=280,407.55
XS Rating Curve= 0 ,0
Exp/Cntr(USF)=0,0
Exp/Cntr=0.3,0.1

Type RM Length L Ch R = 1 ,14603   ,114,114.7,118.8
XS GIS Cut Line= 3
1589384.35607887409849.2822479321588777.90103274410614.182347308
1588784.35956566411017.058217166
#Sta/Elev= 30
       0  647.99    77.6  647.06   103.4  642.43     142  642.03   161.3  636.42
   180.7  633.84   244.1  632.45   251.5  631.31     290  619.13   320.6   614.6
   335.6  606.04   346.2  604.94   463.7  604.94   470.2606.1118     484  615.13
   494.2  618.58   571.9  630.92   848.1  629.47   939.2  631.09   958.7  631.75
  1002.5  640.92  1030.5   640.3  1066.5  635.59  1130.5  636.67  1158.5  641.99
  1193.3  642.87  1222.5  655.52  1294.5  671.18  1342.5  688.67  1379.1  691.39
#Mann= 15 ,-1,0
       0     .08       0      10     .07       0     140     .06       0
     260    .025       0     290      .1       0   335.6    .045       0
   470.2     .08       0     510     .07       0     770     .06       0
     890     .05       0     930     .07       0 1006.15     .06       0
 1106.15     .08       0 1206.15     .05       0 1306.15     .06       0
Bank Sta=335.6,470.2
XS Rating Curve= 0 ,0
Exp/Cntr(USF)=0,0
Exp/Cntr=0.3,0.1

Type RM Length L Ch R = 1 ,14489   ,303.3,256.8,201.9
XS GIS Cut Line= 3
1589303.27796852409774.9533860991588719.01845849410509.634275086
 1588725.4769914410912.510144944
#Sta/Elev= 30
       0  642.16      94  635.23   298.4  630.27     320  624.81   352.1  617.45
   364.9  612.23   372.6607.5272   380.2  605.34   390.5  604.94   513.1  604.97
  521.52  607.56   528.4  613.55   548.9  623.65   570.6   629.3   726.5   629.2
   945.6  631.67   958.4  632.84   993.8  643.12  1037.1  644.95  1089.6  644.11
  1129.6  636.15  1149.6  639.68  1173.6  647.06  1210.4  646.94  1269.6  662.84
  1285.6  664.23  1301.6  662.37  1313.6  664.16  1329.6  663.69  1341.6   665.9
#Mann= 12 ,-1,0
       0     .08       0     320     .07       0     360    .025       0
   372.6    .045       0  521.52     .07       0     640     .05       0
     740     .07       0     800     .05       0     860     .07       0
 1078.68     .06       0 1178.68     .08       0 1268.68     .05       0
Bank Sta=372.6,521.52
XS Rating Curve= 0 ,0
Exp/Cntr(USF)=0,0
Exp/Cntr=0.3,0.1

Type RM Length L Ch R = 1 ,14232   ,776.4,731.2,688.5
XS GIS Cut Line= 5
1588675.68710109409609.5548753931588767.93136336409916.760884855
1588783.14544357410188.2196616091588511.38161211410564.714927988
1588580.65453443410933.459555933
#Sta/Elev= 30
       0  761.73    19.8  756.96    44.9   746.3    74.1  722.46    99.2  697.85
   111.7   693.4   145.1  671.44   216.1  641.01   262.1  637.35   303.8  630.28
   376.6  626.25   408.7  615.69   419.4   607.8   424.7   605.5   436.7  604.88
   540.9  604.94  550.04  607.74   556.9  614.57   560.9  616.34     593  620.83
   976.1  616.03  1007.4  621.59  1032.1   634.8  1051.8  641.83  1117.8   645.5
    1244  648.25  1309.1  654.69    1335  653.73    1362  661.64  1432.2  673.59
#Mann= 9 ,-1,0
       0      .1       0     260     .06       0  360.76      .1       0
   419.4    .045       0  550.04    .025       0  560.76     .05       0
 1136.97     .06       0 1236.97     .08       0 1336.97     .06       0
#XS Ineff= 2 , 0
          368.77  639.29  679.59          638.25
Permanent Ineff=
       F       F
Bank Sta=419.4,550.04
XS Rating Curve= 0 ,0
Exp/Cntr(USF)=0,0
Exp/Cntr=0.3,0.1

Type RM Length L Ch R = 1 ,13501   ,686.3,682.6,678.9
XS GIS Cut Line= 6
1587616.95916873409855.1763185881587686.35010607409926.638774084
1587824.04438448410068.4426243331588191.95375365410447.333926918
1588317.97665208410578.693873324 1588372.9667869410979.718708974
#Sta/Elev= 30
       0  816.67    56.9  796.25   102.1  789.45   125.1  791.24   164.4  783.75
   188.3  773.29   211.2  771.98   262.9  751.52   291.8  748.63   337.6  735.82
   442.4  661.65   464.7  661.21   503.7  644.79   521.3  644.11   548.3  634.79
   583.1  633.57   600.1  626.39   614.2  627.33   648.7  614.65     658  607.77
   670.6  604.88   764.1  604.88   774.6607.9629   810.3  622.78   941.2  631.27
  1009.3  645.57  1081.9  654.16  1146.6  658.46  1231.1  653.26  1412.2  664.93
#Mann= 11 ,-1,0
       0      .1       0  444.14     .06       0  585.39      .1       0
     658    .045       0   774.6      .1       0  825.39     .05       0
  875.39     .06       0  965.39      .1       0 1177.43     .05       0
 1277.43     .06       0 1377.43     .07       0
#XS Ineff= 2 , 0
          608.86  632.08
Permanent Ineff=
       F       F
Bank Sta=658,774.6
XS Rating Curve= 0 ,0
Exp/Cntr(USF)=0,0
Exp/Cntr=0.3,0.1

Type RM Length L Ch R = 1 ,12818   ,505.2,500,494.9
XS GIS Cut Line= 6
1587133.85742459410399.5495776681587354.15652467410599.137105003
1587425.94936009410664.179953918 1587615.8521955410836.229150504
 1588024.6072835411206.5541972521588171.95574209411340.049665168
#Sta/Elev= 30
       0  771.77    31.3  760.73      84  729.89   112.7  723.81   132.5  725.21
   159.6  720.13   208.2  705.83   240.2  691.21   353.9  663.18   449.7   647.6
   461.1  642.75   478.1  644.34   542.8   633.4   591.3  631.51   615.1     618
     648  606.18   656.1  604.88  766.95606.2189   775.4  612.44   783.9  613.89
   972.6  622.51  1030.3   637.7  1143.5  653.06  1171.9  666.31  1210.9  667.12
  1233.7  684.77    1305  719.26  1359.8  753.91  1384.8  765.71  1400.8  769.27
#Mann= 8 ,-1,0
       0      .1       0  367.27     .06       0  404.14      .1       0
     648    .045       0  766.95    .025       0  810.39     .05       0
 1096.64     .06       0 1241.95      .1       0
Bank Sta=648,766.95
XS Rating Curve= 0 ,0
Exp/Cntr(USF)=0,0
Exp/Cntr=0.3,0.1

Type RM Length L Ch R = 1 ,12318   ,491.3,500,508.8
XS GIS Cut Line= 6
1586772.22855468410824.5854730011586930.16918367410945.363446668
1587229.29456967411174.1067555841587427.88406751411325.968984678
1587727.00912543411554.7119655011587884.95008251411675.490267262
#Sta/Elev= 30
       0  696.62   105.6  673.97   185.4   651.3   196.2  650.72   236.5  658.35
   302.8  648.15   347.3   649.7   432.9  642.59   528.6  640.77   553.5  629.08
   567.7  630.93   587.7  627.76   613.4  612.29  634.48606.4008   649.4  604.88
   758.9  606.32   781.7  614.69   807.4  613.12   902.1  618.54   930.1  626.61
    1012  642.03  1072.4  668.32  1109.9  668.88  1125.9  681.95  1138.4  711.73
  1144.1  718.17  1251.1   763.3    1284  768.88  1343.9   787.1  1400.8  811.73
#Mann= 6 ,-1,0
       0      .1       0  634.48    .045       0   758.9    .025       0
  835.39      .1       0 1002.89     .06       0 1163.52      .1       0
Bank Sta=634.48,758.9
XS Rating Curve= 0 ,0
Exp/Cntr(USF)=0,0
Exp/Cntr=0.3,0.1

Type RM Length L Ch R = 1 ,11818   ,488.4,500,512.2
XS GIS Cut Line= 6
1586526.21231443411122.7531837521586659.11624809411271.034383252
1586725.41598426411343.9466390011586791.47195451 411414.89236325
1586857.04039292411481.9066649231587502.55156909412127.417841092
#Sta/Elev= 30
       0  681.01    18.5  673.76    68.9  663.39   104.3  648.92   128.8   643.8
   249.8  648.62   366.2  620.63   483.9  624.75   509.4  630.11   599.9  619.97
   611.5  615.06   628.2  613.35  636.83606.5497   650.5  604.88  770.76606.5924
   803.2  623.59   831.8  646.81   877.1  667.23   888.1  676.28     922  677.26
     928  683.54   939.3  706.28   944.6  711.22   961.6  721.33   995.5  734.19
  1035.1  739.71  1109.3  740.85  1244.4  759.29  1318.6  774.14  1401.3  777.85
#Mann= 5 ,-1,0
       0      .1       0  636.83    .045       0  770.76      .1       0
  835.87     .06       0  973.37      .1       0
#XS Ineff= 2 , 0
          505.78  646.89
Permanent Ineff=
       F       F
Bank Sta=636.83,770.76
XS Rating Curve= 0 ,0
Exp/Cntr(USF)=0,0
Exp/Cntr=0.3,0.1

Type RM Length L Ch R = 1 ,11318   ,520.7,500,477.2
XS GIS Cut Line= 6
1586206.11157668411354.1621697551586534.40521142411826.706172168
1586577.19712059 411888.300209091586634.25278075411970.426029086
1586780.45852509 412180.873114751587005.33865276412504.564068422
#Sta/Elev= 30
       0  697.09    31.6  687.08   129.5  665.57   155.5     653   178.8  647.95
   375.1  638.34   431.4  629.25   460.7  629.59   487.2  619.01   575.4  613.21
   616.6  613.26   631.2  606.02   646.9  604.88   767.7  606.02   777.3  615.33
   801.7  626.54   900.9   639.5   918.6  637.81     950  623.75     977  635.15
   991.6  638.16  1040.3  639.26  1059.8  634.39  1093.9  650.86  1118.2  656.87
  1210.2  655.49  1258.4  660.79  1293.5  660.14    1352  667.52  1400.8  668.26
#Mann= 9 ,-1,0
       0      .1       0  218.83     .08       0  258.83      .1       0
  337.27     .08       0  434.14      .1       0   631.2    .045       0
   767.7    .025       0  820.39      .1       0 1291.95     .06       0
#XS Ineff= 2 , 0
                          909.23          652.99
Permanent Ineff=
       F       F
Bank Sta=631.2,767.7
XS Rating Curve= 0 ,0
Exp/Cntr(USF)=0,0
Exp/Cntr=0.3,0.1

Type RM Length L Ch R = 1 ,10818   ,543.6,500,450.5
XS GIS Cut Line= 6
  1585642.696693411796.6767046751586240.34247933412250.444826007
1586500.35705118412491.9453272521586584.37624009412551.814630091
1586700.51216267412592.086859256  1586832.635258412623.066128001
#Sta/Elev= 30
       0  760.38    36.9  753.77   106.5  732.97   142.4  715.52   167.5  694.95
   224.7  670.69   243.6  670.65   317.3  657.85   418.6  632.95   453.8  628.02
   478.9  630.38     509  616.19   614.7   612.8   631.8   606.2   639.6  604.88
   774.3 606.239   785.8  612.82   822.8  623.03   882.3  628.01  1003.7  645.64
  1077.4  650.49  1113.4   640.8  1144.5   651.8  1159.2  653.41  1193.6  639.21
    1231  633.76  1259.2  638.25  1301.5  652.33  1359.9  652.68  1467.3  667.81
#Mann= 4 ,-1,0
       0      .1       0  527.89     .06       0   631.8    .045       0
   774.3      .1       0
Bank Sta=631.8,774.3
XS Rating Curve= 0 ,0
Exp/Cntr(USF)=0,0
Exp/Cntr=0.3,0.1

Type RM Length L Ch R = 1 ,10318   ,542,500,452.7
XS GIS Cut Line= 6
1585328.22816184412696.1722810121586153.26194485412671.905925334
1586240.48158668412661.0817999991586436.57371417412624.207858011
1586552.48457159 412617.946059511586824.66250493412639.598903343
#Sta/Elev= 30
       0  918.63    15.9  911.06    34.5   893.1    63.9   882.4    95.9  857.26
   115.9  847.13     156  814.82     232  778.84     268  748.32     320  727.68
     336  709.16   364.9  688.36   428.1  663.59   544.1  625.59   564.1  630.82
   588.1  624.91   604.1  614.78   636.2  608.35   648.2  604.88   756.2  604.95
  766.67608.2781   792.2   614.8   824.2  631.88   888.7  642.38  1071.7   648.1
  1108.3  637.76  1208.5  632.54  1260.6  645.36  1332.7  648.97    1502   668.9
#Mann= 6 ,-1,0
       0      .1       0  434.14     .05       0  537.89     .07       0
  635.39    .025       0   636.2    .045       0  766.67      .1       0
Bank Sta=636.2,766.67
XS Rating Curve= 0 ,0
Exp/Cntr(USF)=0,0
Exp/Cntr=0.3,0.1

Type RM Length L Ch R = 1 ,9818    ,1235.7,1214.5,1179.6
XS GIS Cut Line= 6
1585753.23223309413543.600376174 1586193.0797786413172.644425169
1586384.18832026413011.468894511  1586672.045028412768.697726503
1586747.89133301 412704.731319011586856.32484317412679.388193846
#Sta/Elev= 30
       0  873.33   122.6  862.34   134.6   852.1   155.5  824.72   186.9  805.47
   218.3  763.75   244.5  748.83   259.7   722.5   290.9  704.29   461.2  640.94
   485.2  637.89   501.1  630.64   563.1  627.29   629.1607.4408   645.7  604.88
   776.3  607.44   784.8  614.22   813.2  617.58   848.6  631.79   904.4  625.98
   966.4  647.51     998  642.47  1024.1     652  1051.7  649.33  1074.4  654.68
  1092.2  650.98  1115.3  658.48  1144.5   656.3  1190.8  665.65  1412.5  667.75
#Mann= 7 ,-1,0
       0      .1       0  404.14     .07       0  527.89    .025       0
   629.1    .045       0   776.3    .025       0  790.39      .1       0
 1401.17     .06       0
Bank Sta=629.1,776.3
XS Rating Curve= 0 ,0
Exp/Cntr(USF)=0,0
Exp/Cntr=0.3,0.1

Type RM Length L Ch R = 1 ,8604    ,,,
XS GIS Cut Line= 6
1586878.74082218414474.1731212011587255.26078555413760.534539578
 1587294.6927735413687.704858059 1587343.3143954413607.549178476
1587444.60946841413440.5573864821588077.87482122412990.425483592
#Sta/Elev= 30
       0  706.21    47.1  687.49    83.3  685.61   105.8  670.94   268.7  682.53
   294.4  689.32   309.4  687.55   345.8  697.66   404.4  698.62   458.2  661.94
     473   641.6   487.8  629.26   535.5  629.24   570.7  614.88   612.4  612.69
   623.9   607.1     635  604.88  766.82  607.07   870.6  648.41  1207.1  657.24
  1369.5  644.08  1537.8  657.17  1568.5  669.72  1620.2  670.08  1668.9  690.03
  1731.1  698.78  1772.2  720.17  1806.6  731.48  1896.8  742.45  1955.7  744.43
#Mann= 17 ,-1,0
       0     .05       0     110      .1       0     140     .06       0
     220      .1       0     330     .05       0     440     .07       0
     550      .1       0   623.9    .045       0  766.82    .025       0
     780      .1       0 1003.44     .07       0 1120.32      .1       0
 1160.32     .07       0 1258.76     .06       0 1288.76     .07       0
 1528.76     .06       0 1648.76      .1       0
Bank Sta=623.9,766.82
XS Rating Curve= 0 ,0
Exp/Cntr(USF)=0,0
Exp/Cntr=0.3,0.1
LCMann Table=0

Chan Stop Cuts=-1
Use User Specified Reach Order=0
Composite Channel Slope=5
